--- FALLINGRCR.prj (project) ---

Proj Title=FALLINGRCR
Current Plan=p01
Default Exp/Contr=0,0
English Units
Geom File=g01
Flow File=f01
Plan File=p01
BEGIN DESCRIPTION:
END DESCRIPTION:
DSS Export Rating Curves= 0
DSS Export Rating Curve Sorted= 0
DSS Export Volume Flow Curves= 0
DXF OffsetX= 0
DXF OffsetY= 0
DXF ScaleX= 0
DXF ScaleY= 0

--- FALLINGRCR.p01 (plan) ---

Plan Title=Floodplain
Program Version=4.00
Geom File=g01
Flow File=f01
K Sum by GR=0
Std Step Tol=0.01
Critical Tol=0.01
Num of Std Step Trials=20
Max Error Tol=0.3
Flow Tol Ratio=0.001
Split Flow NTrial=30
Split Flow Tol=0.02
Split Flow Ratio=0.02
Log Output Level=0
Friction Slope Method=1
Unsteady Friction Slope Method=2
Unsteady Bridges Friction Slope Method=1
Global Log Level=0
CheckData=False
Run HTab=0
Run UNet=0
Run PostProcess=0
UNET Theta=0
UNET Theta Warmup=0
UNET ZTol=0
UNET ZSATol=0
UNET MxIter=0
UNET MaxInSteps=0
UNET DtIC=0
UNET DtMin=0
UNET MaxCRTS=0
UNET WFStab=0
UNET SFStab=0
UNET WFX=0
UNET SFX=0
UNET DSS MLevel=0
UNET DZMax Abort=0
UNET Convert EG Bridges=0
UNET Use Existing IB Tables=0
UNET Froude Limit=0
UNET Froude Power=0
Write IC File=0
Echo Input=False
Echo Output=False
Write Detailed=0

--- FALLINGRCR.f01 (steady flow) ---

Flow Title=NFF Regression Equation
Program Version=4.10
Number of Profiles= 1
Profile Names=P100yr
River Rch & RM=FALLINGRCR,Main            ,80806.8
679.1446
River Rch & RM=FALLINGRCR,Main            ,80644.1
984.3234
River Rch & RM=FALLINGRCR,Main            ,79185.2
1039.641
River Rch & RM=FALLINGRCR,Main            ,76389.4
1119.403
River Rch & RM=FALLINGRCR,Main            ,72390.6
1426.589
River Rch & RM=FALLINGRCR,Main            ,67482.5
1580.656
River Rch & RM=FALLINGRCR,Main            ,63581.9
2456.726
River Rch & RM=FALLINGRCR,Main            ,56271.9
2911.237
River Rch & RM=FALLINGRCR,Main            ,53726.5
3098.357
River Rch & RM=FALLINGRCR,Main            ,47144
3382.919
River Rch & RM=FALLINGRCR,Main            ,46355.3
3593.804
River Rch & RM=FALLINGRCR,Main            ,43037.2
 3777.96
River Rch & RM=FALLINGRCR,Main            ,34755.2
3952.716
River Rch & RM=FALLINGRCR,Main            ,19052.3
4386.752
River Rch & RM=FALLINGRCR,Main            ,5342.9
4832.067
Boundary for River Rch & Prof#=FALLINGRCR,Main            , 1
Up Type= 0
Dn Type= 3
Dn Slope=0.0016
DSS Import GetInterval= 0
DSS Import GetPeak= 0
DSS Import FillOption= 0

--- FALLINGRCR.g01 (geometry) ---

Geom Title=USGS 10m DEM
Program Version=4.10

River Reach=FALLINGRCR      ,Main
Reach XY= 30
     1892298.122      513656.497     1886813.516      518702.739
     1881058.558      514674.076     1877962.215      514701.307
     1875751.977      511449.362      1874105.99       511568.78
      1873665.74      512588.318     1872902.026      512089.812
     1872918.702      513768.884     1871696.618      513352.009
     1870374.552      514184.995      1870121.62      516895.431
     1868635.623      519282.699     1867909.482      517997.193
     1865500.173        516906.1     1864998.471      518261.692
     1863209.137      517417.212     1862194.651      518181.251
     1859850.769      517657.824     1860162.012      519072.803
     1857198.133      523742.113     1857762.195      525604.274
     1856516.188      527914.962      1858538.88      530852.816
      1857583.62      531068.921       1857642.8      532418.942
     1856349.121      531924.184     1856306.295      533102.882
     1854693.704       533469.95     1853938.408      534834.829

Type RM Length L Ch R = 1 ,80806.8 ,84.6,81.7,78.8
XS GIS Cut Line= 2
     1892201.225      513618.064     1892520.166      513775.448
#Sta/Elev= 24
       0 1016.32     9.6 1012.89    19.2 1009.28    28.8 1005.56    48.1  997.78
    57.7  992.54    67.3  986.85    76.9  983.74    86.5  982.06    96.1  981.36
   105.7  981.44   115.4  982.11     125  983.43   134.6   984.4   144.2  984.13
   153.8  984.05   163.4   984.1   192.2     984   201.9  984.01   230.7  984.37
   269.2  985.01   307.6  985.89   336.4  986.84   355.7  987.67
#Mann= 3 , 0 , 0
       0      .1       0    86.5    .045       0   115.4      .1       0
Bank Sta=86.5,115.4
XS Rating Curve= 0 ,0
Exp/Cntr=0.3,0.1

Type RM Length L Ch R = 1 ,80725.1 ,84.7,81,77.3
XS GIS Cut Line= 3
     1892168.423      513706.609     1892451.757      513803.832
     1892518.423      513846.193
#Sta/Elev= 27
       0 1003.59     9.7 1001.11    19.3  998.25      29  995.19    38.6  991.72
    48.3  988.54      58  986.45    77.3  982.49    86.9981.3321    96.6  980.96
   106.9981.2713     116  982.05   125.6  983.04   135.3  983.68   154.6   984.1
   164.3  984.21   173.9  984.21   183.6     984   202.9     984   212.6  984.13
   280.2  985.46   308.3  986.08   325.9  986.28   334.6  986.29   343.4  986.47
     361  987.58   378.5  988.31
#Mann= 3 , 0 , 0
       0      .1       0    86.9    .045       0   106.9      .1       0
Bank Sta=86.9,106.9
XS Rating Curve= 0 ,0
Exp/Cntr=0.3,0.1

Type RM Length L Ch R = 1 ,80644.1 ,34.1,34.1,34.1
XS GIS Cut Line= 3
     1892153.405      513801.152      1892306.97      513827.474
     1892455.202      513882.102
#Sta/Elev= 21
       0  990.52     9.7   989.6    19.5  988.54    29.2  987.28    48.7   984.2
    68.2  981.54    77.9  980.74    87.6  980.21    97.4  980.64   116.8  983.42
   126.6  983.92   146.1  984.05   165.1  984.03   183.7  984.19     193  984.02
   202.3  984.05   230.2  985.09     258  985.78   267.3  986.11   276.6  986.54
   313.8  988.66
#Mann= 3 , 0 , 0
       0     .06       0    77.9    .045       0    97.4      .1       0
#XS Ineff= 2 , 0
                          160.13           985.6
Permanent Ineff=
       F       F
Bank Sta=77.9,97.4
XS Rating Curve= 0 ,0
Exp/Cntr=0.3,0.1

Type RM Length L Ch R = 1 ,80610   ,124.1,142.5,161
XS GIS Cut Line= 3
     1892146.191      513834.419     1892299.756      513860.741
     1892399.005      513897.544
#Sta/Elev= 21
       0  988.68    29.2  984.84      39  983.96    48.7  983.28    58.4  982.92
    68.2  982.32    77.9  980.69    87.6  979.67    97.4  979.68   104.2980.6904
   107.1  981.12   116.8  983.35   126.6  984.26   136.3  984.24   146.1  984.07
   184.7  984.09   194.3  984.34   232.8  986.22   242.4  986.76     252  987.47
   261.7  988.44
#Mann= 3 , 0 , 0
       0     .06       0    77.9    .045       0   104.2      .1       0
#XS Ineff= 2 , 0
                          126.84          985.54
Permanent Ineff=
       F       F
Bank Sta=77.9,104.2
XS Rating Curve= 0 ,0
Exp/Cntr=0.3,0.1

Type RM Length L Ch R = 1 ,80467.4 ,204.6,216.6,227.9
XS GIS Cut Line= 2
     1892086.082      513828.152     1892224.376      514038.539
#Sta/Elev= 25
       0  994.12    19.4   992.3      29  991.26    38.7  990.07    48.4   988.7
    58.1   987.1    67.8  984.82    77.5  982.88    87.2  981.82   106.5   981.7
   125.9  981.37   145.2  981.29   154.9  981.09   164.6  980.28   166.7980.0426
   174.3  979.18     184  979.34   186.7979.9169   193.7  981.42   203.4  985.23
     213  988.14   222.7  990.21   232.4  994.56   242.1 1001.33   251.8 1006.78
#Mann= 3 , 0 , 0
       0     .06       0   166.7    .045       0   186.7      .1       0
Bank Sta=166.7,186.7
XS Rating Curve= 0 ,0
Exp/Cntr=0.3,0.1

Type RM Length L Ch R = 1 ,80250.8 ,263.4,236.4,209.7
XS GIS Cut Line= 4
     1891945.919      513886.518      1891964.79      513948.314
     1891978.198      514130.361     1892021.613      514193.462
#Sta/Elev= 28
       0  997.87     9.2  996.72    27.7  994.59    46.2   992.3    55.4  991.13
    64.6  989.74    74.2   986.9    83.8  982.12    93.4  978.44    94.5 978.275
     103     977   112.6  977.12   122.3  977.48   141.5  979.72   151.1  980.65
   160.7  981.27   179.9  982.21   199.1  982.91   237.6  983.72   247.2  984.26
   256.7     985   266.3  986.91   275.9  990.81   285.4  995.75     295  999.68
   304.6 1001.64   314.2 1002.73   323.8 1005.98
#Mann= 3 , 0 , 0
       0      .1       0    94.5    .045       0   122.3      .1       0
Bank Sta=94.5,122.3
XS Rating Curve= 0 ,0
Exp/Cntr=0.3,0.1

Type RM Length L Ch R = 1 ,80014.4 ,144.1,158,171.4
XS GIS Cut Line= 4
     1891709.635      514057.923     1891753.493      514102.087
      1891844.89      514132.144     1891922.626      514237.646
#Sta/Elev= 23
       0 1013.24    17.8 1004.67    35.6  995.48    44.5  991.21    53.4  988.49
    71.9  984.14    81.5  980.64    91.1  976.89   100.7  976.05   110.4  977.96
     120  980.65   129.6  982.09   139.2  982.65   177.2   984.6   195.9  985.67
   205.3  986.35   214.6  987.28   233.3   989.6   242.7   990.6   252.1   992.1
   261.4   994.8   280.1 1002.28   289.5 1005.23
#Mann= 3 , 0 , 0
       0      .1       0    91.1    .045       0   110.4      .1       0
Bank Sta=91.1,110.4
XS Rating Curve= 0 ,0
Exp/Cntr=0.3,0.1

Type RM Length L Ch R = 1 ,79856.4 ,244.2,225.2,204.7
XS GIS Cut Line= 2
     1891636.011      514111.455     1891792.955      514317.011
#Sta/Elev= 20
       0 1013.81    19.2 1004.86    38.3   995.7    47.9  991.67    57.5  987.99
      67  983.95    76.6  981.09    86.2  980.65   134.1  979.89   162.8  979.32
   172.4  978.68   182.3977.0357   191.6  975.96   201.2  976.63   210.7  980.84
   220.3  986.59   229.9  989.76   239.5  991.05     249  993.78   258.6  997.64
#Mann= 3 , 0 , 0
       0      .1       0   182.3    .045       0   201.2      .1       0
Bank Sta=182.3,201.2
XS Rating Curve= 0 ,0
Exp/Cntr=0.3,0.1

Type RM Length L Ch R = 1 ,79631.2 ,230.1,251.4,272.5
XS GIS Cut Line= 4
     1891422.318      514239.391     1891542.525      514370.791
     1891632.558      514376.631     1891728.432      514473.478
#Sta/Elev= 30
       0 1008.43    28.1 1003.96    56.2 1000.85    93.7  995.68   121.8  992.26
   131.2  991.31   140.6  990.72     150   990.5   168.7   989.3   178.1     988
   187.1  986.07   196.1  982.73   205.2  978.81   214.3976.0331   223.2  975.41
   232.2  976.65   241.2  978.87   250.3  980.72     278  985.79   287.8   988.1
   297.5  991.06   307.2  994.59   336.4 1005.75   346.2 1008.76   355.9 1009.95
   365.6 1009.51   375.4 1010.27   385.1 1014.89   394.8 1022.82   404.6  1026.7
#Mann= 3 , 0 , 0
       0      .1       0   214.3    .045       0   232.2      .1       0
Bank Sta=214.3,232.2
XS Rating Curve= 0 ,0
Exp/Cntr=0.3,0.1

Type RM Length L Ch R = 1 ,79379.8 ,27.1,44.5,59.2
XS GIS Cut Line= 3
     1891445.208      514529.272     1891448.589      514559.416
     1891496.824       514634.39
#Sta/Elev= 18
       0  982.34     7.6  981.82    15.2  981.29    22.8  980.92    30.3  980.49
    39.2  979.28    48.2   976.7    50.7   976.2    57.1  974.93    65.7  975.53
      66  975.55    68.2976.4177    74.9  979.06    83.8  983.48    92.7   986.1
   101.6  987.67   110.6  988.67   119.5  989.57
#Mann= 3 , 0 , 0
       0     .08       0    48.2    .045       0    68.2     .08       0
Bank Sta=48.2,68.2
XS Rating Curve= 0 ,0
Exp/Cntr=0.3,0.1

Type RM Length L Ch R = 1 ,79335.3 ,32.2,29.4,29.3
XS GIS Cut Line= 2
     1891433.307       514528.95      1891422.49      514684.576
#Sta/Elev= 19
       0  982.24     9.8  981.72    19.5  981.29    29.2  980.92      39  980.31
    48.8  979.05    58.5  976.82    68.2   974.6    72.7  974.34      78  974.04
    87.7  974.34    90.2974.5186    97.5  975.04   107.2  975.85     117   978.9
   126.8  981.11   136.5  982.11   146.2   982.5     156  982.99
#Mann= 3 , 0 , 0
       0     .08       0    68.2    .045       0    90.2     .08       0
Bank Sta=68.2,90.2
XS Rating Curve= 0 ,0
Exp/Cntr=0.3,0.1

Type RM Length L Ch R = 1 ,79305.8 ,121.9,120.6,118.3
XS GIS Cut Line= 2
     1891404.552       514531.79     1891393.735      514687.416
#Sta/Elev= 19
       0  981.89     9.8  981.38    19.5  980.82    29.2  980.24      39  979.44
    48.8  978.14    58.5  976.21    68.2  974.41    74.7  973.97      78  973.74
    87.8  974.21    89.7  974.57    97.5  976.07   107.2  978.34     117  979.41
   126.8  980.04   136.5  980.63   146.2  981.22     156   981.7
#Mann= 3 , 0 , 0
       0     .08       0    68.2    .045       0    87.8     .08       0
Bank Sta=68.2,87.8
XS Rating Curve= 0 ,0
Exp/Cntr=0.3,0.1

Type RM Length L Ch R = 1 ,79185.2 ,152.9,146.7,140.8
XS GIS Cut Line= 3
     1891283.182       514529.32     1891283.289      514617.441
     1891306.796      514688.625
#Sta/Elev= 20
       0   985.9     9.8  983.03    19.6  980.43    29.4  977.84    39.2  975.05
    44.2  974.04      49  973.08    58.8  972.49    59.2   972.5    68.5  972.83
    78.3  973.58    88.1   974.3    97.5  974.76   106.9   975.3   116.2  975.88
   125.6  976.53     135  977.12   144.4  977.75   153.7  978.38   163.1  978.98
#Mann= 3 , 0 , 0
       0      .1       0      49    .045       0    68.5     .08       0
Bank Sta=49,68.5
XS Rating Curve= 0 ,0
Exp/Cntr=0.3,0.1

Type RM Length L Ch R = 1 ,79038.5 ,278.9,274.6,270.4
XS GIS Cut Line= 3
     1891126.178      514529.867     1891165.019      514667.724
     1891169.296      514763.833
#Sta/Elev= 29
       0  997.44     9.6  993.82    19.1  990.21    28.6  986.19    38.2  981.92
    47.7  978.61    57.3  977.01    66.8  976.46    76.4   975.9    85.9  974.51
    93.4  972.96    95.5  972.52     105  971.89   108.4  972.18   110.9972.3937
   114.6  972.71   124.1  974.02   133.7  974.83   143.2  975.12   152.8  975.38
   162.5  975.67   172.1  975.96   181.7  976.27   191.3  976.63     201  976.76
   210.6  976.83   220.2   977.7   229.8  980.02   239.4  983.88
#Mann= 3 , 0 , 0
       0      .1       0    95.5    .045       0   110.9     .08       0
Bank Sta=95.5,110.9
XS Rating Curve= 0 ,0
Exp/Cntr=0.3,0.1

Type RM Length L Ch R = 1 ,78763.9 ,62.6,55.2,41.9
XS GIS Cut Line= 4
     1890846.818      514560.013     1890864.527      514643.867
     1890918.172      514758.971     1890920.777      514791.263
#Sta/Elev= 30
       0  989.38     9.5  985.95      19  982.53    28.6  979.28    38.1  977.24
    47.6  976.64    57.1  976.24    66.7  975.91    76.2  975.65    85.7  975.27
    95.5  974.99   105.2   974.7     115  974.44   124.8  974.14   134.6  973.83
   144.3  973.46   154.1  972.56   161.4  971.25   163.8  970.82   173.6  970.23
   176.4  970.52   178.9970.7736   183.4  971.23   193.2  972.61   202.9  974.35
   212.7   977.7   220.8  981.83   228.9  986.51     237  991.44   245.1  996.25
#Mann= 3 , 0 , 0
       0     .06       0   163.8    .045       0   178.9     .06       0
Bank Sta=163.8,178.9
XS Rating Curve= 0 ,0
Exp/Cntr=0.3,0.1

Type RM Length L Ch R = 1 ,78708.6 ,46.1,45.4,48.5
XS GIS Cut Line= 4
     1890737.977      514574.488     1890742.828       514626.08
      1890885.59      514761.421     1890892.544      514794.208
#Sta/Elev= 25
       0  985.34     8.6  982.01    17.3  979.52    25.9   978.1    51.8  975.54
    61.7  974.45    71.5  973.58    81.3  973.38     101  972.64   110.8  972.53
   120.7  972.64   140.3  973.23     160  973.55   169.8  973.44   179.7  972.84
   189.5  971.13   199.4   970.4   209.2  970.94     219  972.54   238.7  974.65
   248.5  976.84   256.9  980.84   265.3  985.81   273.7  991.15   282.1  996.31
#Mann= 3 , 0 , 0
       0     .06       0   189.5    .045       0   209.2     .06       0
Bank Sta=189.5,209.2
XS Rating Curve= 0 ,0
Exp/Cntr=0.3,0.1

Type RM Length L Ch R = 1 ,78663.3 ,170.6,181.7,191
XS GIS Cut Line= 4
     1890701.518      514571.449     1890709.745       514650.85
     1890838.266       514772.78     1890845.551      514813.006
#Sta/Elev= 27
       0  986.41     8.9  983.21    17.7  980.61    26.6  979.16    53.2  977.71
    89.7  975.93    99.5  975.31   119.2   973.8     129  973.38   148.7  973.26
   158.6  973.49   168.4  973.42   178.2  973.56   188.1  973.43   197.9  971.75
   199.9971.4967   207.8   970.5   217.4  970.52   219.9970.8542   227.5  971.87
   237.3  973.86   247.1  975.69     257  978.32   265.2  982.67   281.5   993.3
   289.7  998.26   297.9 1002.38
#Mann= 3 , 0 , 0
       0     .06       0   199.9    .045       0   219.9     .06       0
Bank Sta=199.9,219.9
XS Rating Curve= 0 ,0
Exp/Cntr=0.3,0.1

Type RM Length L Ch R = 1 ,78481.6 ,191.8,189.3,186.7
XS GIS Cut Line= 4
     1890567.838      514620.928     1890606.032      514734.644
     1890645.963      514829.262     1890675.911      514877.439
#Sta/Elev= 18
       0  980.26    27.7  978.34    46.1   977.3   129.3  973.72   157.3   972.7
   166.6  972.15     176  971.12   185.3     970   194.6   969.8  199.57 971.053
     204  972.17   213.3  975.51   222.7   977.5   232.1   978.8   241.6  980.97
     251  984.77   260.5  989.71   279.4  999.88
#Mann= 3 , 0 , 0
       0     .06       0     176    .045       0  199.57      .1       0
Bank Sta=176,199.57
XS Rating Curve= 0 ,0
Exp/Cntr=0.3,0.1

Type RM Length L Ch R = 1 ,78292.2 ,251.6,247.6,243.6
XS GIS Cut Line= 3
      1890357.11      514723.804     1890419.981      514802.216
     1890502.631      514949.856
#Sta/Elev= 24
       0  999.41     9.1  994.86    18.3  990.39    27.4  986.65    45.7  979.46
    54.8  976.76      64  975.52    91.4  973.91   109.9  972.67   147.5  970.54
   156.9  970.11   166.3  969.84   175.7  969.46   188.8 968.725   194.5  968.44
   203.9   968.5   208.8  969.18   213.3  969.81   222.7  974.33   232.1  979.78
   241.5  983.97   250.9  986.45   260.3  988.27   269.7  991.33
#Mann= 3 , 0 , 0
       0     .07       0   188.8    .045       0   208.8      .1       0
Bank Sta=188.8,208.8
XS Rating Curve= 0 ,0
Exp/Cntr=0.3,0.1

Type RM Length L Ch R = 1 ,78044.6 ,497.9,483.3,468.9
XS GIS Cut Line= 2
     1890170.033       514889.28     1890335.605      515095.625
#Sta/Elev= 22
       0 1008.72    19.6  999.83    29.4  995.27    39.2  989.77    58.8  976.38
    68.6  971.09    78.4     969    88.2  968.92   117.6  968.99   156.8  969.27
   176.4   969.3   186.2  968.56   191.7967.7969     196   967.2   205.8  966.65
   211.7968.1033   215.6  969.06   225.4  974.79   235.2  980.69     245  985.29
   254.8  987.09   264.6  987.89
#Mann= 3 , 0 , 0
       0     .07       0   191.7    .045       0   211.7      .1       0
Bank Sta=191.7,211.7
XS Rating Curve= 0 ,0
Exp/Cntr=0.3,0.1

Type RM Length L Ch R = 1 ,77561.3 ,302.4,312.8,323.1
XS GIS Cut Line= 4
     1889795.414      515085.955     1889814.164      515216.511
     1890000.969      515265.122     1890071.108        515355.4
#Sta/Elev= 30
       0 1007.48    28.3  999.37    37.7  996.04    47.1  991.88    56.5  987.04
      66  982.72    75.4  980.01   103.6  975.27     113  973.89   122.5  972.77
   131.9  971.87   141.6  971.24   170.5  969.71   189.8  968.52   208.8964.0918
   218.8  963.18   228.8963.8428   238.1  965.07   247.7  965.93     267  966.64
   286.3  967.58   305.6  968.96   315.3  969.99   324.9  971.47   334.4  973.61
   372.6  982.96   401.1  990.26   410.7  992.29   420.2  993.77   439.2  994.77
#Mann= 3 , 0 , 0
       0      .1       0   208.8    .045       0   228.8      .1       0
Bank Sta=208.8,228.8
XS Rating Curve= 0 ,0
Exp/Cntr=0.3,0.1

Type RM Length L Ch R = 1 ,77248.5 ,358.8,367.1,374.8
XS GIS Cut Line= 4
     1889522.358        515252.2     1889649.556      515411.403
     1889734.901      515484.439     1889797.269      515569.784
#Sta/Elev= 30
       0 1005.57    19.4 1001.57    38.8     997    48.5  994.29    58.2  990.94
    67.9  986.79    77.6  983.18    87.3  981.25   155.3  973.69   194.1  970.23
   213.1  967.78   222.5   966.8   231.9  966.01   241.2  965.84   250.6     965
   259.9  962.84   269.3  961.82   278.8961.9722     288  963.09   297.4  964.63
   306.8   965.1   344.9  965.48   354.5  966.58   364.2  969.87   373.8  975.22
   383.4  979.36     393  980.96   402.6  982.07   412.2  984.53   421.8  989.02
#Mann= 3 , 0 , 0
       0     .07       0   259.9    .045       0   278.8      .1       0
Bank Sta=259.9,278.8
XS Rating Curve= 0 ,0
Exp/Cntr=0.3,0.1

Type RM Length L Ch R = 1 ,76881.4 ,501.8,492,482.2
XS GIS Cut Line= 4
     1889260.312      515558.157     1889406.561      515607.881
     1889484.365      515748.865     1889573.284      515861.184
#Sta/Elev= 30
       0  997.63    38.6  987.02    57.9   981.5    67.6  979.02    77.2  977.15
    96.5  974.21   125.5  969.38   135.2  967.99   144.8  966.86   163.9  965.57
   173.4  964.69   182.9  962.35   192.4959.1813   201.8   958.3   211.3  958.41
   230.2   963.4   239.7   964.5   249.2  964.96   258.7  965.66   277.6  968.21
   315.5  972.03   334.6   973.6   363.2  975.52   382.4  977.21   401.4  978.65
     411  979.08   420.6  979.27   430.1  979.82   439.6  981.49   458.8  988.34
#Mann= 3 , 0 , 0
       0     .07       0   192.4    .045       0   211.3      .1       0
Bank Sta=192.4,211.3
XS Rating Curve= 0 ,0
Exp/Cntr=0.3,0.1

Type RM Length L Ch R = 1 ,76389.4 ,98.7,97.8,96.7
XS GIS Cut Line= 2
     1889065.918      515964.559     1889309.841       516142.51
#Sta/Elev= 22
       0  991.84     9.7  989.75    19.5  987.06      39  980.42    48.7   977.5
    68.2  972.49    77.9  969.82    87.7  966.48   107.1  958.84   116.9  956.96
   126.6  956.91   136.4  958.22   146.1  960.12   155.8  961.07   175.3  961.13
   185.1  961.32     224  962.44   253.2  963.18     263  963.54   272.7  965.21
   282.5   968.9   301.9   978.5
#Mann= 3 , 0 , 0
       0      .1       0   107.1    .045       0   136.4      .1       0
Bank Sta=107.1,136.4
XS Rating Curve= 0 ,0
Exp/Cntr=0.3,0.1

Type RM Length L Ch R = 1 ,76291.6 ,37.7,37.8,37.7
XS GIS Cut Line= 2
     1888999.553      516044.359     1889274.075       516226.65
#Sta/Elev= 24
       0  978.32    19.4  973.91    29.1  972.36    48.5  970.05    58.2  968.98
    67.8  967.74    77.5  966.72    87.2  965.33    96.9  963.79   106.6   961.2
   116.3  958.46     126   956.5   135.7  956.35   145.4  957.17   155.1  958.92
   164.8  960.24   174.5  960.45   184.2  960.15   193.8  960.18   261.7  961.32
   271.4  962.37   281.1  965.44   319.8  984.55   329.5  989.14
#Mann= 3 , 0 , 0
       0      .1       0     126    .045       0   145.4      .1       0
Bank Sta=126,145.4
XS Rating Curve= 0 ,0
Exp/Cntr=0.3,0.1

Type RM Length L Ch R = 1 ,76253.8 ,267.7,255.3,241.2
XS GIS Cut Line= 2
     1888978.532      516075.684     1889253.054      516257.976
#Sta/Elev= 25
       0  976.77     9.7  975.63    29.1  972.93    48.5  970.04    67.8  967.52
   106.6  961.92   116.3  959.96     126  957.84   127.1957.6812   135.7  956.44
   145.4  957.03   147.1957.3245   155.1  958.71   164.8  959.77   174.5  959.86
   184.2  959.81   203.5  959.91     252  960.62   261.7  960.88   271.4  962.47
   281.1  966.95   290.8  973.61   300.5  978.98   310.2  983.22   329.5  990.48
#Mann= 3 , 0 , 0
       0     .08       0   127.1    .045       0   147.1      .1       0
Bank Sta=127.1,147.1
XS Rating Curve= 0 ,0
Exp/Cntr=0.3,0.1

Type RM Length L Ch R = 1 ,75998.5 ,198.4,202.8,206.8
XS GIS Cut Line= 4
     1888807.365      516381.974     1888868.789      516392.135
     1889179.144      516392.597     1889237.335      516395.368
#Sta/Elev= 30
       0 1005.96    17.8  998.36    35.6     991    62.3  980.57      72  975.83
    81.7  969.86    91.4  963.48     101  959.03   110.8  957.91   130.2     958
   149.6  957.85   227.1  957.95   236.8  957.47   246.5  956.46   256.2  955.88
   265.9  956.21   285.3  960.54   304.7  961.18   314.4  961.82   324.1  963.15
   333.8   966.8   343.5  972.96   353.2  979.81   362.9  986.43   372.6  991.78
   382.3  994.91     392  996.53   411.4  999.43   421.2  1001.2   430.9 1003.41
#Mann= 3 , 0 , 0
       0     .08       0   246.5    .045       0   265.9      .1       0
Bank Sta=246.5,265.9
XS Rating Curve= 0 ,0
Exp/Cntr=0.3,0.1

Type RM Length L Ch R = 1 ,75795.6 ,325.7,332.9,339.9
XS GIS Cut Line= 3
     1888810.874      516543.092     1889108.548      516600.046
     1889304.366      516563.969
#Sta/Elev= 30
       0  987.15     9.8   981.8    19.6  975.67    29.3  969.27    39.1  962.61
    48.9  956.89    58.7  954.41    78.2  954.27   127.1  954.24   166.2  955.17
   185.8  955.46   234.6  955.32   244.4  955.07   254.2  954.48     264  954.13
   268.6955.2825   273.7  956.56   283.5  961.47   293.3  964.97   312.6  966.86
   331.5  971.65     341  973.04   350.5  974.67     360  976.66   407.4  988.56
   416.8  990.67   445.3  996.34   473.7 1002.47   483.2 1004.59   502.2  1009.1
#Mann= 3 , 0 , 0
       0      .1       0   244.4    .045       0   268.6      .1       0
Bank Sta=244.4,268.6
XS Rating Curve= 0 ,0
Exp/Cntr=0.3,0.1

Type RM Length L Ch R = 1 ,75462.7 ,191.7,183.9,174.8
XS GIS Cut Line= 2
     1888721.203      516703.576     1889010.664       516864.29
#Sta/Elev= 28
       0  985.27     9.7  981.82    29.2  975.31      39  972.17    48.7  969.47
    58.4  966.66    68.2  963.22    77.9  957.17    87.6  950.63    97.4  948.29
   107.1  948.89   116.8  949.85   126.6  950.19   175.3  950.38   194.8  950.53
   204.5  950.74   214.2  951.29   233.7  953.21   243.4   954.5   253.2  956.73
   262.9  960.91   272.7  966.52   282.4   971.1   292.1     973   301.9  974.55
   311.6   978.9   321.4  984.98   331.1  989.96
#Mann= 3 , 0 , 0
       0      .1       0    87.6    .045       0   107.1      .1       0
Bank Sta=87.6,107.1
XS Rating Curve= 0 ,0
Exp/Cntr=0.3,0.1

Type RM Length L Ch R = 1 ,75278.8 ,536.3,547.4,558.2
XS GIS Cut Line= 4
     1888589.179      516798.068      1888781.94      516908.413
     1888893.659      516923.065     1888990.269      516995.408
#Sta/Elev= 30
       0  984.89     9.7  982.37    19.3   979.2    38.6  970.86    48.3  968.36
    57.9  967.92    67.6  967.91    77.3  967.33    86.9  966.17   135.2  959.71
   144.8  958.59   193.1   954.4   222.1  951.68   250.3   949.3   269.1  947.05
   278.4   946.8   287.8  946.93   297.2   948.3   306.6  950.06   325.4  952.86
   334.8  955.38   344.1  960.19   362.6  973.61   371.9  977.52   390.5  981.68
   399.8   985.6   409.1  991.23   418.3  996.56   427.6 1000.87   455.5 1011.07
#Mann= 3 , 0 , 0
       0      .1       0   269.1    .045       0   287.8      .1       0
Bank Sta=269.1,287.8
XS Rating Curve= 0 ,0
Exp/Cntr=0.3,0.1

Type RM Length L Ch R = 1 ,74731.4 ,412.2,412.8,413.3
XS GIS Cut Line= 3
     1888392.385       517238.43     1888542.776      517345.201
     1888644.338       517450.67
#Sta/Elev= 27
       0  995.37     9.7  992.36    19.4  988.72    29.1  984.06    38.8  978.64
    48.5  973.01      68  961.39    77.7  955.82    87.4  951.06    97.1  946.42
   106.8  942.95   116.5  941.59   126.2  942.11   128.3 942.582   135.9  944.29
   145.6  946.89   155.3  948.25     165  949.34   184.4  951.12   194.2  951.89
   213.7  952.83   252.8  954.26   272.3  954.85   301.6  955.89   311.3  956.64
   321.1  957.94   330.9  959.46
#Mann= 3 , 0 , 0
       0      .1       0   106.8    .045       0   128.3      .1       0
Bank Sta=106.8,128.3
XS Rating Curve= 0 ,0
Exp/Cntr=0.3,0.1

Type RM Length L Ch R = 1 ,74318.6 ,60.5,56.1,51.5
XS GIS Cut Line= 4
       1888161.8      517556.755     1888195.887      517600.281
     1888261.962      517649.575     1888287.658      517675.271
#Sta/Elev= 24
       0  953.49     9.2  949.95    18.4  947.68    27.6  946.58    36.9  945.88
    46.1  945.17    55.3  944.47    64.4  943.82    73.6  942.92    82.8  941.45
    89.5 940.515    91.9  940.18      92  940.18   101.1  939.95     107  940.75
   109.5941.0938   110.2  941.19   119.4  943.55   128.6  945.29   137.7  946.46
   146.8  947.82   155.9  949.35     165  951.11   174.1  953.39
#Mann= 3 , 0 , 0
       0      .1       0    89.5    .045       0   109.5      .1       0
Bank Sta=89.5,109.5
XS Rating Curve= 0 ,0
Exp/Cntr=0.3,0.1

Type RM Length L Ch R = 1 ,74262.5 ,37,37,37
XS GIS Cut Line= 3
     1888095.385      517622.645     1888233.305      517688.196
     1888283.123       517689.77
#Sta/Elev= 27
       0   946.4     9.5  945.99    19.1  945.83    28.6  945.58    38.2  945.11
    47.7  944.43    57.3  943.82    66.8  943.51    76.4  943.41    85.9  943.11
    95.4  941.83   104.4940.0769     105  939.96   106.9  939.81   114.5   939.2
   121.9  940.02   124.1  940.26   124.4 940.338   133.6  942.73   143.2  945.42
   152.7  947.61     161  949.18   169.3  951.06   177.6  953.08   185.9  954.87
   194.2  956.21   202.6  957.54
#Mann= 3 , 0 , 0
       0      .1       0   104.4    .045       0   124.4      .1       0
Bank Sta=104.4,124.4
XS Rating Curve= 0 ,0
Exp/Cntr=0.3,0.1

Type RM Length L Ch R = 1 ,74225.5 ,81.2,95.9,110.4
XS GIS Cut Line= 3
     1888096.159      517663.944     1888234.079      517729.495
     1888283.897      517731.068
#Sta/Elev= 26
       0  945.12     9.5  944.75    19.1  944.28    28.6  943.73    38.2  943.26
    47.7  943.04    57.3  943.16    66.8     943    76.4  941.35    85.9  939.54
    86.2939.5186    88.7  939.34    95.4  938.86   103.7  940.05     105  940.24
   114.5  942.98   124.1  946.05   133.6  948.39   143.2  950.71   152.7  953.33
     161  955.07   169.3  956.73   177.6  958.46   185.9  960.51   194.2  962.96
   202.6   965.6
#Mann= 3 , 0 , 0
       0     .07       0    86.2    .045       0     105      .1       0
Bank Sta=86.2,105
XS Rating Curve= 0 ,0
Exp/Cntr=0.3,0.1

Type RM Length L Ch R = 1 ,74129.6 ,202.4,200.1,197.5
XS GIS Cut Line= 4
     1888078.337      517673.368     1888104.684      517742.655
     1888131.335      517792.502     1888171.342      517835.535
#Sta/Elev= 25
       0  944.84     9.3  944.47    18.5     944    27.8  943.47    37.1     943
    46.3  942.52    55.6  942.12    64.9  941.69    74.1  941.25    83.6  940.63
      93  939.28    96.9938.5975    99.4  938.16   102.4  937.64   111.8  937.45
   114.4  938.22   116.9938.9626   121.2  940.24   130.6  945.34   140.4   950.5
   150.2  955.22     160  959.73   169.8  964.21   179.6  968.53   189.4  972.64
#Mann= 3 , 0 , 0
       0     .07       0    96.9    .045       0   116.9      .1       0
Bank Sta=96.9,116.9
XS Rating Curve= 0 ,0
Exp/Cntr=0.3,0.1

Type RM Length L Ch R = 1 ,73929.5 ,337.9,338.5,338.2
XS GIS Cut Line= 2
     1887902.042      517801.798     1888020.098      517973.673
#Sta/Elev= 25
       0  944.24     9.5   943.5      19  942.76    28.4  942.13    37.9  941.45
    47.4  940.83    56.9  939.94    66.4  938.43    75.8  936.66    82.9  935.17
    85.3  934.66    94.8  933.38    97.9  933.32   104.3   933.2   113.7  934.05
   123.2   935.6   132.7  935.91   142.2  936.18   151.6  938.29   161.1  942.34
   170.6  947.13   180.1  951.89   189.6  956.74     199  961.46   208.5  965.97
#Mann= 3 , 0 , 0
       0     .08       0    85.3    .045       0   113.7      .1       0
Bank Sta=85.3,113.7
XS Rating Curve= 0 ,0
Exp/Cntr=0.3,0.1

Type RM Length L Ch R = 1 ,73591   ,347.3,347.8,347.4
XS GIS Cut Line= 2
     1887626.521      517942.781     1887796.877      518195.602
#Sta/Elev= 23
       0  978.14     9.8  974.56    39.3  964.19    49.2  960.45    78.7  948.72
    88.5  944.27    98.3  939.29   108.2  935.66     118  935.01   137.7  934.93
     177     935   186.8  934.19   189.9933.6973   196.7  932.62   206.5  932.12
   209.9932.5733   216.4  933.44   226.2  936.79     236  940.69   265.5  951.48
   275.4  955.24   285.2  959.15   304.9   967.4
#Mann= 3 , 0 , 0
       0      .1       0   189.9    .045       0   209.9      .1       0
Bank Sta=189.9,209.9
XS Rating Curve= 0 ,0
Exp/Cntr=0.3,0.1

Type RM Length L Ch R = 1 ,73243.3 ,247.6,246.8,245.7
XS GIS Cut Line= 3
     1887360.679      518144.604     1887493.058      518342.087
     1887549.481       518400.68
#Sta/Elev= 27
       0  970.46     9.5  967.46      19  964.64    28.5  961.01      38  957.88
    57.1  951.18    66.6  947.38    76.1  943.13    95.1  931.73   102.2929.2114
   104.6  928.36   114.1  927.89   122.2928.8284   133.1  930.18   142.6  930.84
   161.7  931.93   180.7  933.39   209.2  936.08   237.8  938.55   246.8  939.17
   264.9  940.25   273.9   940.9   282.9  941.56     292  942.51     301  944.36
     310  947.36   319.1  951.07
#Mann= 3 , 0 , 0
       0      .1       0   102.2    .045       0   122.2      .1       0
Bank Sta=102.2,122.2
XS Rating Curve= 0 ,0
Exp/Cntr=0.3,0.1

Type RM Length L Ch R = 1 ,72996.5 ,248.9,238.4,225.6
XS GIS Cut Line= 3
     1887139.607       518267.63     1887301.867      518488.794
     1887384.628      518564.492
#Sta/Elev= 30
       0   986.8     9.8  982.13    19.6  977.68    29.4   973.4    39.2  969.31
    58.8  961.54    88.2  950.26      98  945.55   107.8  938.79   117.6  932.27
   127.4  928.39   137.2  927.08     147  927.48   148.8927.8159   156.7  929.29
   166.5  930.41   176.3   931.1   225.3  933.84   244.9  934.75   254.7  934.96
   274.3   935.1     293  935.38   302.3  935.79   311.7  936.54     321  937.39
   330.4  938.58   349.1  942.17   367.8  946.08   377.1  947.45   386.5   948.7
#Mann= 3 , 0 , 0
       0      .1       0   127.4    .045       0   148.8      .1       0
Bank Sta=127.4,148.8
XS Rating Curve= 0 ,0
Exp/Cntr=0.3,0.1

Type RM Length L Ch R = 1 ,72758.2 ,206.1,205.6,204.6
XS GIS Cut Line= 5
     1886960.908       518445.44     1887015.369        518508.5
     1887165.854      518584.459     1887631.639      518686.215
     1887676.785      518803.737
#Sta/Elev= 30
       0  962.34    18.5  955.47    27.8  952.46    83.3  935.71    92.7  933.19
   111.4  927.29   120.8  925.13   130.2   924.2   148.9  924.43   167.6  927.52
     177  928.18   223.8  929.92     320  932.75   368.6  934.83   397.8  937.79
   407.6  939.31   446.5  947.78   475.7  952.93   485.4  955.42   602.2  988.26
   611.9  990.29   621.6  991.47   631.4  993.69   650.8 1000.78   660.6 1003.84
   728.7 1023.25   767.4 1025.49   796.4 1024.89   825.5  1022.6   854.6 1018.57
#Mann= 3 , 0 , 0
       0      .1       0   120.8    .045       0   148.9      .1       0
Bank Sta=120.8,148.9
XS Rating Curve= 0 ,0
Exp/Cntr=0.3,0.1

Type RM Length L Ch R = 1 ,72552.6 ,66.5,67.1,66.1
XS GIS Cut Line= 4
     1886845.537      518512.083     1886857.675       518626.93
     1887061.508      518737.299     1887114.976      518930.574
#Sta/Elev= 30
       0  951.69     9.6  949.39    48.1  942.47    57.7  938.25    67.4  931.93
      77  928.22    86.6  928.07   115.5  931.38   125.1  931.14   134.8  929.88
   163.8  924.78   171.6924.0488   183.1  923.63   192.8   924.3   212.1  927.68
   221.7  928.31   289.3  927.09   337.6  927.79   347.3  927.63   356.8  928.06
   385.5  930.79     395  932.94   404.6  936.36   433.2  947.66   461.9  958.27
   471.4  961.02     481  963.46   519.2  972.57   528.7  975.22   547.8  981.17
#Mann= 3 , 0 , 0
       0      .1       0   171.6    .045       0   192.8     .08       0
#XS Ineff= 2 , 0
          116.01  934.58   315.3          934.12
Permanent Ineff=
       F       F
Bank Sta=171.6,192.8
XS Rating Curve= 0 ,0
Exp/Cntr=0.3,0.1

Type RM Length L Ch R = 1 ,72485.5 ,63.7,94.9,127.6
XS GIS Cut Line= 4
      1886790.27       518528.41     1886801.901       518659.31
     1887030.195      518782.923     1887073.164      518922.246
#Sta/Elev= 30
       0  948.14    37.6   942.2    46.9  939.29    56.3  933.08    65.7  928.34
    75.1  928.93    93.9  932.02   103.3  932.72   112.6  932.79     122     932
   131.4  930.54     141  929.57   160.3  928.02   179.5  924.31   189.1  922.98
   198.7  922.33   208.3  922.72     218   923.6   237.2  926.44   246.8  927.43
   275.6  927.08   304.5   927.7   333.3  929.65   362.2  932.47     391  933.98
   400.8  936.47   459.1  956.02   478.5   962.1   507.7  970.35   536.8  978.02
#Mann= 3 , 0 , 0
       0     .08       0   189.1    .045       0   208.3     .08       0
#XS Ineff= 2 , 0
          110.06   935.4
Permanent Ineff=
       F       F
Bank Sta=189.1,208.3
XS Rating Curve= 0 ,0
Exp/Cntr=0.3,0.1

Type RM Length L Ch R = 1 ,72390.6 ,557,590.1,621.6
XS GIS Cut Line= 4
     1886775.696      518526.588     1886775.696      518654.111
     1886746.548      518765.237     1886774.482      518926.159
#Sta/Elev= 30
       0  947.79    39.2  941.26      49  938.51    58.9  933.39    68.7  928.96
    78.5  928.19    98.1  929.94   107.9  930.43   127.5  930.32   146.7     928
   156.2  925.75   165.8  922.45   175.4  920.82     185  922.02   194.5   925.1
   204.1  927.64   223.3  931.36   232.8  932.24   242.4  932.37   261.6  931.66
   271.2  931.69   280.8  932.94     300   938.7   309.7  940.86   319.3  941.77
   348.1  943.41   376.9  943.97   386.5  944.75   396.1  947.07   405.7  950.04
#Mann= 3 , 0 , 0
       0      .1       0   165.8    .045       0     185      .1       0
#XS Ineff= 2 , 0
          117.56  931.72
Permanent Ineff=
       F       F
Bank Sta=165.8,185
XS Rating Curve= 0 ,0
Exp/Cntr=0.3,0.1

Type RM Length L Ch R = 1 ,71800.5 ,410.8,372.6,334.2
XS GIS Cut Line= 4
     1886603.134      518322.095     1886462.186      518474.356
     1886273.822      518456.853     1886191.283      518746.581
#Sta/Elev= 30
       0  981.82    47.2  970.18    75.4  962.71   113.2  954.09   122.6  951.49
     132  947.86   169.8  928.46   179.2  925.23   188.6  924.18   226.4  923.37
   302.1  920.74   311.5  920.17   328.3917.8495   339.9  916.69   349.4  918.05
   368.3  924.09   377.7  926.33   387.2  927.61   396.7  928.22   464.7  935.79
   513.3  942.35     523  943.21   532.7   943.5   581.3   943.7   600.7  944.22
   610.4   946.5   620.2  951.71   629.9  955.46   649.3  958.26   697.9  966.54
#Mann= 3 , 0 , 0
       0      .1       0   328.3    .045       0   349.4      .1       0
Bank Sta=328.3,349.4
XS Rating Curve= 0 ,0
Exp/Cntr=0.3,0.1

Type RM Length L Ch R = 1 ,71427.9 ,583.7,592.5,600.8
XS GIS Cut Line= 3
       1886083.9      518088.448     1886085.394      518496.677
     1886028.035       518663.01
#Sta/Elev= 30
       0 1023.85     9.7 1020.27    77.8  988.77    87.5  985.56   106.9  981.09
   116.6  978.13   126.4   974.3   136.1  969.97     175  951.78   184.7  946.68
   194.4  940.08   204.1  931.33   213.8  921.56   223.6   914.9   233.3  913.35
     243   915.4   252.7  918.96   262.4  921.85   272.2  923.44   340.2  931.26
   437.6  941.92   447.3  942.83   457.1  943.27   525.5  943.76   535.3  944.73
   545.1  948.78   554.8  955.26   564.6  960.59   574.4  963.86   584.2  966.69
#Mann= 3 , 0 , 0
       0      .1       0   223.6    .045       0     243      .1       0
Bank Sta=223.6,243
XS Rating Curve= 0 ,0
Exp/Cntr=0.3,0.1

Type RM Length L Ch R = 1 ,70835.4 ,445.6,447.3,449
XS GIS Cut Line= 3
     1885675.263      518170.244     1885614.055      518448.086
     1885536.819      518637.052
#Sta/Elev= 30
       0   959.7     9.8  957.07    29.4  951.39      49  946.33    68.7  942.47
    88.3  939.27    98.1  938.01   117.7     936   137.4  933.66   166.8  929.48
   186.4  926.94   235.4  921.74   255.1     920   284.5  918.99   294.2  918.24
   313.7  916.04   323.4  914.51   340.7909.6532   342.8  909.06   352.6   907.7
   362.3  909.01     372   913.6   391.4  926.62   401.2  932.91   410.9  938.52
   420.6  942.13   430.3   946.1     440  953.06   449.8  957.54   488.6  971.47
#Mann= 3 , 0 , 0
       0      .1       0   340.7    .045       0   362.3      .1       0
Bank Sta=340.7,362.3
XS Rating Curve= 0 ,0
Exp/Cntr=0.3,0.1

Type RM Length L Ch R = 1 ,70388.1 ,442.6,442,441.2
XS GIS Cut Line= 3
     1885458.083      518082.902     1885302.861      518396.346
     1885295.362      518586.811
#Sta/Elev= 30
       0  969.85    19.4  961.55    38.9  953.82    48.6   948.4    58.3  939.14
    77.7  916.79    87.4  907.49    94.6904.1647    97.1  903.01   106.9  902.38
   114.6903.1911   116.6   903.4   126.3  905.65     136  907.39   165.2  910.91
     204  915.95   213.8   916.7   242.9  918.05   262.3  919.69   310.9  924.34
   340.1  926.68   359.3  928.53   397.4  932.84     407  934.21   445.1  942.15
   483.2  950.87   492.7  953.48   502.3  956.77   530.8  968.82   540.4  972.18
#Mann= 3 , 0 , 0
       0      .1       0    94.6    .045       0   114.6      .1       0
Bank Sta=94.6,114.6
XS Rating Curve= 0 ,0
Exp/Cntr=0.3,0.1

Type RM Length L Ch R = 1 ,69946   ,354.3,358,361.8
XS GIS Cut Line= 3
     1885041.245      517916.581     1885018.322      518029.861
     1884941.419      518200.298
#Sta/Elev= 27
       0  938.62     9.6  934.63    19.3  930.99    28.9  927.46    38.5  924.33
    57.8  919.13    67.4  916.73    86.7  912.16    96.3  909.75   105.9  907.77
   115.6  906.32   125.4     905   145.1     903   154.9  900.96   164.8  898.21
   174.6  896.93   184.5  897.97   194.3  902.32   204.2  908.02     214   912.3
   223.8   914.5   233.7  915.31   253.4  916.22   263.2  917.27     273  919.23
   292.7  924.13   302.6  926.51
#Mann= 3 , 0 , 0
       0      .1       0   164.8    .045       0   184.5      .1       0
Bank Sta=164.8,184.5
XS Rating Curve= 0 ,0
Exp/Cntr=0.3,0.1

Type RM Length L Ch R = 1 ,69588   ,356.1,356.5,356.8
XS GIS Cut Line= 2
     1884801.916      517748.723     1884679.674      517931.712
#Sta/Elev= 28
       0  953.15     9.6  947.19    19.1  939.38    28.7  928.72    38.3  917.25
    47.8  906.73    57.4   899.4      67  895.85    69.6895.4014    72.1  894.97
    76.5  894.21    86.1  893.92    87.1  894.03    89.6894.2946    95.7  894.94
   105.2   896.6   114.8  897.57   124.4  898.29     134  899.15   143.5   900.1
   153.1  900.98   162.7  901.65   172.2  901.96   181.8  902.19   191.4  902.32
   200.9  902.36   210.5  902.44   220.1  902.47
#Mann= 3 , 0 , 0
       0      .1       0    69.6    .045       0    89.6      .1       0
Bank Sta=69.6,89.6
XS Rating Curve= 0 ,0
Exp/Cntr=0.3,0.1

Type RM Length L Ch R = 1 ,69231.5 ,244,246.4,248.5
XS GIS Cut Line= 3
     1884550.952       517510.41     1884481.981      517590.983
     1884384.625      517731.953
#Sta/Elev= 25
       0  950.01    19.3  941.34    28.9   936.9    38.6  932.18    57.8  922.21
    77.1  912.36    96.4  901.92   106.1  897.74   115.6  895.66   134.6  893.96
   144.1  892.62   153.6  890.95   163.2  890.06   172.7  890.78   182.2  892.82
   191.7  894.48   201.2  895.47   210.8  896.05   220.3  896.92   229.8  898.44
   239.3  900.14   248.8  901.72   258.4  903.18   267.9  904.38   277.4  905.38
#Mann= 3 , 0 , 0
       0      .1       0   153.6    .045       0   172.7      .1       0
Bank Sta=153.6,172.7
XS Rating Curve= 0 ,0
Exp/Cntr=0.3,0.1

Type RM Length L Ch R = 1 ,68985.1 ,167.8,140,112.2
XS GIS Cut Line= 3
     1884447.042      517328.641     1884318.919      517420.036
     1884221.546      517534.492
#Sta/Elev= 26
       0  935.78     9.8  931.32    19.7  926.63    29.5  921.81    39.3  917.13
      59  907.99    68.8  903.22    78.7  898.68    88.5  895.79    98.4  894.89
   108.2  894.78   137.7  894.12   157.4  893.77   166.8  892.98   176.2   890.1
   185.6  886.76   194.8  886.33   204.3  887.22   213.7  888.44   223.1  889.05
   251.3  889.96   260.7  890.43   270.1  892.03   279.5  894.08   298.3  898.39
   307.6  900.93
#Mann= 3 , 0 , 0
       0      .1       0   185.6    .045       0   204.3      .1       0
Bank Sta=185.6,204.3
XS Rating Curve= 0 ,0
Exp/Cntr=0.3,0.1

Type RM Length L Ch R = 1 ,68845.1 ,78.6,61.1,54.7
XS GIS Cut Line= 4
     1884278.525      517068.335     1884168.589      517271.413
     1884213.859      517417.473     1884185.022       517514.76
#Sta/Elev= 30
       0  904.56     9.6  900.41    19.2  896.61    28.9  893.48    38.5  891.32
    48.1  890.75      77   890.3   125.1  888.67   134.7  888.44   192.4  888.42
   230.9  888.88     250  888.55   278.7  888.84   288.3  888.12   307.4  885.09
   316.9  884.39   326.5  884.74     336  885.84   345.6  886.81   355.2   887.2
   374.3  886.96   402.3  887.12   411.5  887.98   420.7  889.74     430  891.87
   448.4  896.39   457.6  898.99   466.9  902.11   476.1  905.37   485.3  908.44
#Mann= 3 , 0 , 0
       0      .1       0   307.4    .045       0   326.5      .1       0
#XS Ineff= 2 , 0
          140.23   895.6
Permanent Ineff=
       F       F
Bank Sta=307.4,326.5
XS Rating Curve= 0 ,0
Exp/Cntr=0.3,0.1

Type RM Length L Ch R = 1 ,68784   ,192.2,248.9,294.7
XS GIS Cut Line= 4
     1884239.082      517030.087     1884120.756       517250.06
     1884174.568      517416.619     1884145.731      517513.905
#Sta/Elev= 30
       0  892.42     9.6  890.87    19.2  890.36    86.5  889.61   144.1  888.73
   163.3  888.32   182.5  888.46   201.7  888.37     221   888.7   230.6  888.76
   259.5  888.54     279  887.74   288.7  887.14   298.4  886.24   317.8  884.79
   327.6  884.02   337.3  883.86     347  884.23   366.5  886.57   376.2  886.87
   385.9  886.79   405.4  887.51   415.1  887.68   424.8  888.76     434   891.5
   443.3  894.51   452.5  897.73   498.6   915.4   507.8  918.52   526.3  924.18
#Mann= 3 , 0 , 0
       0      .1       0   317.8    .045       0     347      .1       0
#XS Ineff= 2 , 0
           86.26  895.33
Permanent Ineff=
       F       F
Bank Sta=317.8,347
XS Rating Curve= 0 ,0
Exp/Cntr=0.3,0.1

Type RM Length L Ch R = 1 ,68535   ,152.3,150.8,149.3
XS GIS Cut Line= 3
     1884235.174      517011.504     1884151.269      517056.655
     1883935.297      517137.926
#Sta/Elev= 21
       0  893.54     9.5  890.87    19.1  890.13    57.2  889.56   124.1  888.91
   172.2  888.24   191.4  888.05     201  887.87   210.7  887.21   223.4884.7332
   229.9   883.5   239.5  883.85   243.4884.8188   249.1  886.23   258.7  889.32
   268.4   893.2     278  898.06   287.6  903.25   306.8  913.26   316.4  918.18
     326  922.92
#Mann= 3 , 0 , 0
       0      .1       0   223.4    .045       0   243.4      .1       0
Bank Sta=223.4,243.4
XS Rating Curve= 0 ,0
Exp/Cntr=0.3,0.1

Type RM Length L Ch R = 1 ,68384.2 ,79.5,96,114.2
XS GIS Cut Line= 2
     1884175.422      516869.963     1883863.657      517011.752
#Sta/Elev= 27
       0  891.22     9.8  888.64    19.6  887.84    29.4  887.64    39.1  887.71
    48.9  887.92    58.7  888.34    68.5   887.9    88.1  887.35     137  886.88
   146.8   886.7   166.4  886.16   176.1  885.81   185.9  885.62   205.5  885.62
   215.3  884.92   224.4883.2208   234.8  881.65   244.4881.9241   254.4  883.47
   264.2   885.2     274  886.61   283.8  889.22   293.6  894.64   322.9  912.82
   332.7  918.79   342.5  923.72
#Mann= 3 , 0 , 0
       0      .1       0   224.4    .045       0   244.4      .1       0
Bank Sta=224.4,244.4
XS Rating Curve= 0 ,0
Exp/Cntr=0.3,0.1

Type RM Length L Ch R = 1 ,68288.2 ,41.6,42.2,41.6
XS GIS Cut Line= 4
     1884172.859      516854.588     1884021.675      516904.983
     1883816.678      516870.817     1883666.348       516982.71
#Sta/Elev= 30
       0  893.39     9.4  890.04    18.8  888.93    46.9  889.32    56.2  889.02
    65.6  888.41    84.4  887.64   131.2  887.14   159.4  886.54   206.6   884.7
   244.4  883.66   253.8  882.73   263.3  881.24   272.7  880.15   282.2  879.79
   291.6  880.36   310.5  883.47     320  884.16   367.2   883.3   385.9  883.29
   395.3  883.46     414  884.65   432.8  886.25   442.2  887.98   451.5  890.86
   460.9  894.78   479.6  903.05   498.4  911.89   535.8  930.35   554.6  939.25
#Mann= 3 , 0 , 0
       0      .1       0   263.3    .045       0   291.6      .1       0
Bank Sta=263.3,291.6
XS Rating Curve= 0 ,0
Exp/Cntr=0.3,0.1

Type RM Length L Ch R = 1 ,68246   ,251.5,232.3,212.5
XS GIS Cut Line= 4
     1884158.339      516821.276     1884007.154      516871.671
     1883802.158      516837.505     1883651.827      516949.399
#Sta/Elev= 30
       0  901.53     9.4  897.73    18.8  894.66    28.1  892.67    46.9  890.65
    56.2  889.87    65.6  889.26    84.4  888.49   140.6  887.66     216  884.28
   244.4  883.97   253.8  883.12     272880.0677   282.2  879.35     292879.7827
   310.5   882.8     320  883.52   329.4  883.54   385.9  882.58   395.3  882.59
   404.7  882.77   423.4  883.66   451.5  884.15   460.9  884.63   470.3  885.61
   479.6  888.56     489  892.27   498.4  896.47   517.1   905.2   554.6  923.38
#Mann= 3 , 0 , 0
       0      .1       0     272    .045       0     292      .1       0
Bank Sta=272,292
XS Rating Curve= 0 ,0
Exp/Cntr=0.3,0.1

Type RM Length L Ch R = 1 ,68013.8 ,394.8,369.7,344.5
XS GIS Cut Line= 4
     1883903.802      516461.678     1883831.199       516616.28
     1883590.328      516754.652     1883569.829      516927.191
#Sta/Elev= 30
       0  954.72      38  942.77    56.9   936.1    66.4  932.54    85.4  925.04
   142.3     902   151.8  898.28   161.3   894.9   170.8  892.05   180.4  889.75
     190  888.24   209.1  885.76   218.7  883.17   227.5880.1358   228.3  879.86
   237.8  878.42   247.5878.9093   266.6  882.36   276.2  882.52   285.8  882.44
   333.6   881.1     372  881.04   391.1   881.3   429.4  882.45   477.6  883.14
   545.1  884.69   554.8  886.58   564.4  890.87   574.1  895.82   622.3  921.12
#Mann= 3 , 0 , 0
       0      .1       0   227.5    .045       0   247.5      .1       0
Bank Sta=227.5,247.5
XS Rating Curve= 0 ,0
Exp/Cntr=0.3,0.1

Type RM Length L Ch R = 1 ,67644   ,147.6,161.6,175.9
XS GIS Cut Line= 3
     1883456.951      516509.821      1883469.91      516778.906
     1883461.525      516878.765
#Sta/Elev= 25
       0  931.33     9.6   923.6    19.2  914.68    28.9  906.27    38.5  898.34
    48.1  890.59    57.7  884.19    67.4   881.3    96.2  879.46   125.1  877.93
   134.7  877.29   144.3  876.23   149.5875.7775   153.9   875.4   163.6  875.47
   169.5876.3369   182.8  878.32   192.4     879   221.3  880.31   259.8  882.24
   305.8  884.67   342.3  886.48   351.4   887.1   360.5  889.31   369.6  893.31
#Mann= 3 , 0 , 0
       0      .1       0   149.5    .045       0   169.5      .1       0
Bank Sta=149.5,169.5
XS Rating Curve= 0 ,0
Exp/Cntr=0.3,0.1

Type RM Length L Ch R = 1 ,67482.5 ,529.6,529.7,529.4
XS GIS Cut Line= 4
     1883354.809      516521.059      1883343.89      516599.867
     1883256.536      516732.322     1883138.323      516847.686
#Sta/Elev= 29
       0  925.93     8.8  918.94    17.7  910.63    35.4  893.52    44.2  885.22
      53  881.14    61.9  880.47   107.6  878.32   116.9  877.76   126.2  876.84
   135.6  875.52   144.9  874.79   154.2  875.55   163.6  877.47   172.9  878.77
   182.2  879.46   238.2  883.03   247.9  883.58   286.8  885.49   296.5  885.72
   306.2  885.74     316  887.43   325.7  890.49   335.4  894.04   345.1  896.82
   364.5   901.7   374.2  903.92   393.7  908.21   403.4  909.81
#Mann= 3 , 0 , 0
       0      .1       0   135.6    .045       0   154.2      .1       0
Bank Sta=135.6,154.2
XS Rating Curve= 0 ,0
Exp/Cntr=0.3,0.1
