HEC-RAS study FALLINGRCR.prj: FALLINGRCR

--- FALLINGRCR.g01 (geometry) --- (continued)

Type RM Length L Ch R = 1 ,66952.7 ,567.3,567.1,566.7
XS GIS Cut Line= 3
     1883042.234      516296.313     1882890.125       516425.13
     1882777.046      516604.582
#Sta/Elev= 30
       0  934.41     9.5  930.74      19  926.47    28.5  921.89      38  917.01
      57  907.04    66.4  901.97    75.9  897.15    85.4  892.57    94.9  888.26
   104.4  884.57   113.9  882.64   123.4  881.67   142.4  880.16   199.3  876.18
   228.2  874.06   247.5  872.47   257.2  870.81   266.8  868.96   276.5  868.94
   286.1  870.82   295.7  870.82     300869.9094   305.4  868.77     315  868.65
     320870.3064   324.7  871.86   334.3  878.73     344   886.1   411.4  929.96
#Mann= 3 , 0 , 0
       0      .1       0     300    .045       0     320      .1       0
Bank Sta=300,320
XS Rating Curve= 0 ,0
Exp/Cntr=0.3,0.1

Type RM Length L Ch R = 1 ,66385.6 ,570.6,572,573.2
XS GIS Cut Line= 2
     1882593.542      516068.906     1882407.505      516394.143
#Sta/Elev= 26
       0  939.34    19.2  930.27    38.4  921.36      48  916.68    57.6  911.07
    67.2  905.03    76.9   899.1    86.5  893.47   105.7  882.69   115.3  875.62
   124.7869.3729   124.9  869.24   134.5  866.37   144.1   866.6   153.7  868.03
   163.3  869.39   192.2  870.48   259.4  872.48   278.6  872.98   288.2  872.88
   297.8  872.88   307.4  876.82     317  882.67   336.3  894.82   355.5  907.04
   374.7  919.37
#Mann= 3 , 0 , 0
       0      .1       0   124.7    .045       0   153.7      .1       0
#XS Ineff= 2 , 0
                          277.34          877.47
Permanent Ineff=
       F       F
Bank Sta=124.7,153.7
XS Rating Curve= 0 ,0
Exp/Cntr=0.3,0.1

Type RM Length L Ch R = 1 ,65813.6 ,382.1,391.3,400.7
XS GIS Cut Line= 3
     1882110.231      515877.932     1881960.784      516109.392
      1881955.53       516191.23
#Sta/Elev= 25
       0  895.53     9.8  889.78    19.7  884.36    29.5  879.49    39.4  875.41
    49.2  872.39      59  870.78    68.9  870.25    98.4  869.22   157.4  866.64
   167.3   865.5   177.1  863.29   180.4862.6527     187  861.38   196.8  861.07
   206.6  862.36   216.5  864.75   226.3  866.08     246  866.96   275.5  868.45
   302.8  870.12     312  870.82   321.1  872.43   330.2  875.72   357.5   888.8
#Mann= 3 , 0 , 0
       0      .1       0   180.4    .045       0   206.6      .1       0
Bank Sta=180.4,206.6
XS Rating Curve= 0 ,0
Exp/Cntr=0.3,0.1

Type RM Length L Ch R = 1 ,65422.2 ,506.6,504.9,503.5
XS GIS Cut Line= 3
     1881900.321      515649.057     1881585.217      515856.956
     1881449.454      515956.681
#Sta/Elev= 30
       0  905.92    48.4  870.61    58.1  865.72    67.8  864.08    87.1  862.94
   106.5  862.33   125.8  862.14   154.9   861.5   164.6   861.1   174.4860.1022
   183.9  859.24   193.6  859.13   203.3  860.05     213  861.36   222.6  861.95
   300.1  863.91   309.8  865.32   319.4   869.7   329.1  875.76   338.8  882.12
   367.8  901.56   377.5  907.94   396.2  919.41   405.6   924.8   414.9  929.96
     443  944.99   461.7  954.89   480.4  964.62   527.2  988.27     546  997.48
#Mann= 3 , 0 , 0
       0      .1       0   174.4    .045       0   203.3      .1       0
Bank Sta=174.4,203.3
XS Rating Curve= 0 ,0
Exp/Cntr=0.3,0.1

Type RM Length L Ch R = 1 ,64917.3 ,292.5,290.4,288.8
XS GIS Cut Line= 3
     1881653.951      515209.619     1881347.701      515445.036
     1881281.034      515512.397
#Sta/Elev= 29
       0   933.4     9.7  928.35      29  917.96    57.9  902.04   115.9  870.26
   125.5  865.38   135.2  862.98   144.8  861.82   173.8   859.1   193.1  857.01
   197.8856.5726   202.8  856.11   212.4  856.06   217.8856.7635   222.1  857.32
   231.8  859.66   241.4  860.87   251.1  861.09   270.4   861.2   299.4  861.49
     309  861.66     338  862.38   347.6  863.05   357.3  866.21     367  871.34
   376.6  877.14   395.8  888.49   462.1  928.12     481   939.3
#Mann= 3 , 0 , 0
       0      .1       0   197.8    .045       0   217.8      .1       0
Bank Sta=197.8,217.8
XS Rating Curve= 0 ,0
Exp/Cntr=0.3,0.1

Type RM Length L Ch R = 1 ,64626.9 ,303.3,313.4,322.5
XS GIS Cut Line= 4
     1881557.288      514966.726     1881390.565      515059.556
     1881269.564      515174.091     1881134.707      515204.572
#Sta/Elev= 30
       0  928.46    38.2  906.77    66.8  889.59    76.3  884.03    85.9  878.91
    95.4  874.24   114.5  865.45     124   861.8   133.6  859.85   143.1  859.26
   162.2  858.85   200.6  858.93   210.4  858.15   220.2  856.11   224.6854.9622
     230  853.56   239.8  853.47   244.6853.8833   249.6  854.31   259.4  855.68
   269.2  856.52   308.4  858.55     328  859.72   385.1  863.88   394.3  864.81
   403.5   866.9   412.7  870.28     422  874.24   440.4  882.51   495.7  908.36
#Mann= 3 , 0 , 0
       0      .1       0   224.6    .045       0   244.6      .1       0
Bank Sta=224.6,244.6
XS Rating Curve= 0 ,0
Exp/Cntr=0.3,0.1

Type RM Length L Ch R = 1 ,64313.5 ,202.6,188.5,173.2
XS GIS Cut Line= 4
     1881356.435      514793.078      1881269.63      514852.757
     1881107.954       514904.84      1881042.85      514954.753
#Sta/Elev= 24
       0  876.55     9.6  866.67    19.2  859.34    28.7  856.93    38.3  856.64
    47.9  856.56    95.8  856.43   105.3  856.31   133.6  855.76     162  854.97
   190.3  853.98   199.7  853.15   209.1  851.24   218.6  850.43     228  851.21
   237.4  853.44   246.9  855.06   256.3  855.71   284.3  856.61   293.4   857.6
   302.5  860.82   311.7  866.17   329.9  877.63   357.2  895.13
#Mann= 3 , 0 , 0
       0      .1       0   209.1    .045       0     228      .1       0
Bank Sta=209.1,228
XS Rating Curve= 0 ,0
Exp/Cntr=0.3,0.1

Type RM Length L Ch R = 1 ,64125   ,50.2,49.2,49.4
XS GIS Cut Line= 5
     1881299.368      514321.882     1881208.772       514455.82
     1881150.425      514661.818     1881040.298       514803.13
     1880948.707      514889.088
#Sta/Elev= 30
       0  859.99    57.1  858.89   142.7  856.88   171.4  856.39   239.6  855.47
     259  854.94   268.8  854.48   278.5  853.96     298  852.71   307.7  852.25
   336.9  851.81   375.8  851.75   404.1  851.26   413.5  850.75     423  849.69
   432.4  848.95   441.8  849.18   444.6  849.74   451.2  851.06   460.7  852.27
   470.1  852.89   507.8  853.81     555  855.24     584  856.02   593.6  856.73
   603.3  859.87   612.9  865.83   632.3  879.61   670.9  907.57   680.6  914.43
#Mann= 3 , 0 , 0
       0      .1       0     423    .045       0   444.6      .1       0
#XS Ineff= 2 , 0
          307.86  858.13
Permanent Ineff=
       F       F
Bank Sta=423,444.6
XS Rating Curve= 0 ,0
Exp/Cntr=0.3,0.1

Type RM Length L Ch R = 1 ,64075.8 ,223.7,219,213.7
XS GIS Cut Line= 5
     1881276.451      514260.076     1881163.427      514431.122
     1881116.133      514623.491     1881009.311      514775.515
     1880919.121      514867.571
#Sta/Elev= 30
       0   860.5    48.8   859.9   146.4  857.94   185.5  857.43   214.4  856.29
   261.6  855.89     271  855.44   280.5  854.57   299.4  852.14   308.8   851.4
   337.1  850.58   365.4  850.52   384.2  851.19   412.9  851.29     452  850.74
   464.3 849.375   471.6  848.55   481.3  848.59   484.3 849.049   500.9  851.57
   510.7  852.02   569.4  853.33   625.7  854.95   634.9  857.46   644.2  862.54
   653.4  869.42   671.8  884.47     681  891.77   699.4  905.18   717.8  917.68
#Mann= 3 , 0 , 0
       0      .1       0   464.3    .045       0   484.3      .1       0
#XS Ineff= 2 , 0
          350.14   860.4
Permanent Ineff=
       F       F
Bank Sta=464.3,484.3
XS Rating Curve= 0 ,0
Exp/Cntr=0.3,0.1

Type RM Length L Ch R = 1 ,63856.8 ,130.8,127.9,125.2
XS GIS Cut Line= 4
     1880837.562      514310.771     1880947.362      514567.683
     1880927.146      514642.715     1880852.554      514834.624
#Sta/Elev= 30
       0  907.72     9.6  902.82    19.3  897.59    38.5  886.48    48.2  880.77
    77.1  862.51    86.7  857.44    96.3   855.2   144.5   855.1   202.3   855.4
   279.4  854.35   337.7  853.18   376.7  852.86   386.5  852.16   406.1  848.17
   415.9  847.78   425.7  848.68   435.5  850.22   445.3  849.94   455.2  848.38
     465  847.29   474.8  847.85   484.6   853.2   504.2   872.5     514  881.82
   523.8  890.96   533.6  899.55   543.4  907.27   553.2  914.08     563  919.95
#Mann= 3 , 0 , 0
       0      .1       0   455.2    .045       0   474.8      .1       0
Bank Sta=455.2,474.8
XS Rating Curve= 0 ,0
Exp/Cntr=0.3,0.1

Type RM Length L Ch R = 1 ,63728.9 ,147.4,147,146.7
XS GIS Cut Line= 4
     1880750.966      514393.772     1880801.965      514569.554
     1880753.137       514752.93     1880748.796      514828.885
#Sta/Elev= 30
       0  883.35     9.6  879.52    28.9  872.11    57.8  861.34    67.4  857.92
    77.1  855.74    86.7  855.21    96.3  854.96     183  853.53     221   852.6
     240  852.04   249.4  851.84   258.9  851.76   268.4  850.79   277.9   848.8
   287.4   847.9   296.9  848.05   306.4  847.74   313.7 846.864   315.9   846.6
   325.4  846.08   334.8  847.57   344.3  850.92   353.8  853.09   363.3  854.42
   372.8  858.67   410.8   883.7   420.4  889.92   429.8  896.12   448.9  908.47
#Mann= 3 , 0 , 0
       0      .1       0   313.7    .045       0   334.8      .1       0
Bank Sta=313.7,334.8
XS Rating Curve= 0 ,0
Exp/Cntr=0.3,0.1

Type RM Length L Ch R = 1 ,63581.9 ,567,562.9,558.1
XS GIS Cut Line= 5
     1880707.128      514362.625     1880689.455       514516.11
     1880636.973      514618.482     1880602.312      514756.186
     1880600.142      514838.651
#Sta/Elev= 30
       0  898.03     9.7  895.06    48.3  881.77    96.6  866.55   125.5  857.03
   135.2  854.39   144.8  853.05   164.1  851.93   183.3  851.42   221.6   851.3
   240.8  850.64   250.4  851.05   269.5  852.77     279  852.42   288.5  851.57
   297.9  849.54   307.4  846.34   316.9  844.08   326.3  843.69   335.8  845.61
   345.3  848.05   354.7  848.83   373.7  848.69   383.1  849.05   392.6  851.23
   402.1   856.1   420.7  869.19   457.4  896.63   475.7  908.99     494   920.3
#Mann= 3 , 0 , 0
       0      .1       0   307.4    .045       0   335.8      .1       0
#XS Ineff= 2 , 0
          268.77  856.83
Permanent Ineff=
       F       F
Bank Sta=307.4,335.8
XS Rating Curve= 0 ,0
Exp/Cntr=0.3,0.1

Type RM Length L Ch R = 1 ,63019   ,358.3,370.8,383
XS GIS Cut Line= 2
     1880118.235      514506.698     1880103.586      514877.875
#Sta/Elev= 25
       0  873.95     9.8  869.69    19.6  865.96    29.3  862.73    48.9  856.75
    58.6  853.59    68.4  850.69    78.2  848.97      88  846.91    97.8  843.88
   107.5  842.44   117.2842.9842   127.1  844.42   136.9  845.27   146.6  845.36
   234.6  844.74   273.7   844.7   283.5  846.51   293.3  851.58     303  858.02
   312.8  863.92   342.1  880.17   351.9  885.38   361.7  890.38   371.5  895.24
#Mann= 3 , 0 , 0
       0      .1       0    97.8    .045       0   117.2      .1       0
Bank Sta=97.8,117.2
XS Rating Curve= 0 ,0
Exp/Cntr=0.3,0.1

Type RM Length L Ch R = 1 ,62648.2 ,370.8,374.2,377.5
XS GIS Cut Line= 3
     1879926.808      514418.258      1879854.91      514528.082
     1879705.526      514757.122
#Sta/Elev= 28
       0  904.73     9.4  899.26    28.1  888.54    46.9  878.32    65.6  868.31
      75  863.17    84.4  857.89    93.8  852.88   103.1  849.87   112.5  848.94
   170.3  846.76   228.9  845.35   248.5  845.06   277.8  844.48   287.5  844.16
   297.3  843.17     303842.0856   307.1   841.3   316.8  840.37   326.6  841.35
   336.4     845   346.1  849.95   355.9   854.2   365.6  858.61   375.4  863.51
   385.2  868.91     395  874.99   404.7  881.46
#Mann= 3 , 0 , 0
       0      .1       0     303    .045       0   326.6      .1       0
Bank Sta=303,326.6
XS Rating Curve= 0 ,0
Exp/Cntr=0.3,0.1

Type RM Length L Ch R = 1 ,62274   ,135.8,171.1,209.3
XS GIS Cut Line= 3
     1879564.883      514299.284     1879467.555      514457.867
     1879366.249      514571.091
#Sta/Elev= 21
       0  879.17     9.8  873.88    19.6  869.17    29.4  864.77      49  856.18
    58.8  851.67    68.6  848.13    78.3  846.78    88.1  846.55   117.5  846.36
   195.6  846.38   205.1  845.58   214.6  843.24     224  839.49   233.6  838.17
   242.5   838.1   252.5   838.8     262  843.35   271.5  849.62     281  855.42
     338  887.88
#Mann= 3 , 0 , 0
       0      .1       0     224    .045       0   252.5      .1       0
Bank Sta=224,252.5
XS Rating Curve= 0 ,0
Exp/Cntr=0.3,0.1

Type RM Length L Ch R = 1 ,62102.9 ,54.1,53.6,47.3
XS GIS Cut Line= 4
     1879478.112      514292.535     1879335.459      514404.234
     1879227.201      514397.282     1879121.922      514464.819
#Sta/Elev= 30
       0  860.51     9.5  855.75    19.1  851.21    28.6  847.55    38.1  846.16
    76.3  843.52    85.8  843.17    95.4  843.06   114.4  843.11     143  842.86
   152.6  842.97   171.6  843.46   181.2   842.9   190.2   841.8   208.3  838.68
   217.3   838.1   262.5  838.17   271.6  838.87   280.6  840.01   289.7  840.83
   308.9  843.96   318.5  846.07   328.2  847.76   337.8   849.3   347.4  851.05
     357  853.47   366.6   855.7   376.3   857.8   395.5  861.62   414.7  865.12
#Mann= 3 , 0 , 0
       0      .1       0   208.3    .045       0   271.6      .1       0
#XS Ineff= 2 , 0
           121.1  847.02
Permanent Ineff=
       F       F
Bank Sta=208.3,271.6
XS Rating Curve= 0 ,0
Skew Angle= 45
Exp/Cntr=0.3,0.1

Type RM Length L Ch R = 1 ,62049.3 ,223.7,189.5,157.6
XS GIS Cut Line= 5
     1879449.677      514270.152     1879313.609      514376.424
      1879205.35      514369.472     1879115.357      514427.203
      1879100.12      514457.828
#Sta/Elev= 30
       0  862.54    19.2  852.88    28.8  849.04    38.4  847.22    67.1  845.21
    76.7  844.72   115.1  843.67   163.1  842.77   181.7  842.25   190.7  841.61
   208.8  839.46   217.8  838.54   226.9  838.04     245     838     254     838
     263  838.24   272.1   838.1   281.1  838.66   290.8  840.07   300.6  841.11
   310.3  841.45     320  841.29   329.7  840.91   339.4  840.88   349.2  841.08
   358.9  841.62   378.3  844.09     388  845.72   413.7  855.26   422.3  858.27
#Mann= 3 , 0 , 0
       0      .1       0   217.8    .045       0   281.1      .1       0
#XS Ineff= 2 , 0
          115.58   847.6
Permanent Ineff=
       F       F
Bank Sta=217.8,281.1
XS Rating Curve= 0 ,0
Skew Angle= 45
Exp/Cntr=0.3,0.1

Type RM Length L Ch R = 1 ,61859.8 ,260.8,227.6,194.3
XS GIS Cut Line= 4
     1879436.766        514014.9     1879170.588      514176.792
     1879058.357      514298.955     1879094.112      514510.506
#Sta/Elev= 30
       0  935.04    19.5  925.96    38.9  915.61    48.7  909.94    68.2  897.83
    97.4  878.98   116.8  867.44   126.6  862.52   136.3  859.35   175.2  854.86
   194.7   853.4   223.9  852.59   282.3  852.32   321.3  850.71   331.1  849.77
   340.8  848.18   350.6  846.07   370.1  840.58   379.8  838.41   389.6     838
   409.1  838.23   428.6  841.75   438.4  842.19     536  839.77   584.7  840.12
   594.5  840.34   604.2   841.1     614  843.65   623.7  847.98     692   882.9
#Mann= 3 , 0 , 0
       0      .1       0   379.8    .045       0   409.1      .1       0
Bank Sta=379.8,409.1
XS Rating Curve= 0 ,0
Exp/Cntr=0.3,0.1

Type RM Length L Ch R = 1 ,61632.2 ,230.8,229.3,227.7
XS GIS Cut Line= 3
     1878849.151      514166.372     1878978.492      514317.413
      1879073.11      514511.858
#Sta/Elev= 30
       0  928.39     9.5  922.73    18.9  916.99    37.9  905.55    47.4   898.8
    56.8   888.5    66.3  876.18    75.8  863.63    85.2  851.54    94.7   841.8
   104.2  837.71   113.6  837.42   123.1  837.93   132.6  839.46     142  840.31
   151.5  840.39   218.5  839.44   228.3   839.4     248  839.58   277.5   839.5
   287.3  839.64   297.2  839.61     307  839.84   326.6  840.88   336.5  841.51
   346.3   843.4   356.1  847.76     366  852.89   395.4  868.34   415.1  878.55
#Mann= 3 , 0 , 0
       0      .1       0   104.2    .045       0   123.1      .1       0
Bank Sta=104.2,123.1
XS Rating Curve= 0 ,0
Exp/Cntr=0.3,0.1

Type RM Length L Ch R = 1 ,61402.9 ,183.4,157.3,132.1
XS GIS Cut Line= 2
     1878660.548      514309.766     1878922.398      514576.622
#Sta/Elev= 28
       0  931.47    29.5  913.62    39.4  907.74    49.2  901.77      59  895.53
    68.9   888.2    78.7  880.08   108.2  855.42   118.1  848.05   127.9  842.05
   137.7  838.13   147.6  836.49   157.4  835.95   167.3  835.81   177.1  837.22
   186.9  839.27   196.8  840.66   206.6  840.71   236.1  840.15   265.6  840.27
   285.3  840.76   295.2  841.18   314.8  842.14   324.7  842.83   334.5  844.67
   344.4  849.04     364  859.48   373.9  864.66
#Mann= 3 , 0 , 0
       0      .1       0   147.6    .045       0   177.1      .1       0
Bank Sta=147.6,177.1
XS Rating Curve= 0 ,0
Exp/Cntr=0.3,0.1

Type RM Length L Ch R = 1 ,61245.6 ,70.8,67.9,65.4
XS GIS Cut Line= 4
     1878502.188      514495.001     1878570.198      514547.612
     1878781.928      514529.647     1878865.337      514595.091
#Sta/Elev= 30
       0  860.07    28.7   845.4    38.2  841.57    47.8  840.08    57.3  839.48
      86  838.42     115  837.95   124.6  837.71   134.3  837.22   143.9   836.3
   153.6  835.09   163.2  834.05   172.9   833.5   182.6  833.46   192.7833.8167
   201.9  834.49   221.2  836.84   230.9  837.93   240.5  838.74   250.2  839.25
   259.8   839.5   308.1  839.88     337   840.4   346.7  840.64   356.3  841.04
   365.9  841.64   375.6  842.79   385.2  846.26   394.9  851.07   404.5  856.16
#Mann= 3 , 0 , 0
       0      .1       0   163.2    .045       0   192.7      .1       0
Bank Sta=163.2,192.7
XS Rating Curve= 0 ,0
Exp/Cntr=0.3,0.1

Type RM Length L Ch R = 1 ,61177.7 ,168.2,207.7,245.8
XS GIS Cut Line= 4
     1878448.419      514517.587     1878539.527      514595.863
      1878752.54      514575.332     1878834.666      514643.342
#Sta/Elev= 30
       0  855.24     9.2  850.26    18.5  845.82    27.7  842.32      37  840.66
    55.4  839.02    64.7  838.51    73.9  838.26   129.8   837.3   139.6  837.04
   149.3  836.46     159  835.53   168.8   834.4   178.5  833.44   188.2  832.83
   197.9  832.67   207.8  832.84   217.4  833.23   227.1   833.9     266  837.07
   285.5  838.39   295.2  838.91   304.9  839.29   334.1  840.06   372.9  840.63
   382.6  841.19   392.3  844.13     402  848.88     431  864.97   440.8  870.33
#Mann= 3 , 0 , 0
       0      .1       0   178.5    .045       0   217.4      .1       0
Bank Sta=178.5,217.4
XS Rating Curve= 0 ,0
Exp/Cntr=0.3,0.1

Type RM Length L Ch R = 1 ,60970   ,371,380.9,390.8
XS GIS Cut Line= 3
     1878387.407      514512.256       1878472.1      514775.315
     1878635.068       514893.37
#Sta/Elev= 30
       0  864.23    28.6  846.08    38.1  841.87    47.6  840.08    76.2  837.28
    85.8  836.95   123.9  836.84     162  837.63   171.5  836.73   181.1  834.03
   190.6  832.24   200.1  832.18   209.6  832.65   228.7  836.37   238.2  837.81
   257.3  839.28   295.5  840.49   305.1  841.55   314.7   845.4   324.3  852.67
   333.8  860.51   343.4  867.93     353  874.79   362.6  880.91   372.2  885.69
   381.8  888.28   400.9  892.18   429.7  903.67   448.8  909.86   477.6  918.64
#Mann= 3 , 0 , 0
       0      .1       0   181.1    .045       0   209.6      .1       0
Bank Sta=181.1,209.6
XS Rating Curve= 0 ,0
Exp/Cntr=0.3,0.1

Type RM Length L Ch R = 1 ,60589.1 ,300.9,324.7,348.4
XS GIS Cut Line= 4
     1878135.908        514459.8     1878090.157      514590.797
     1878050.758      514897.418     1878020.457      515111.709
#Sta/Elev= 30
       0  890.68    18.5  878.68    27.8  871.29    46.2  855.05    55.5  847.23
    64.8  840.54      74  836.58    83.2   835.7     245  835.88   254.7  834.65
   264.4  831.51     274  829.55   283.7  830.01     303  830.05   312.6  831.48
     332   844.1   389.9   884.3   409.3  896.88   428.6  908.33   438.2  913.32
   467.6  927.22   477.4  932.33   487.2  938.23   536.4   973.5   546.3  979.37
   556.1  984.41     566  988.43   585.6  995.42   634.8 1014.68   664.3 1025.21
#Mann= 3 , 0 , 0
       0      .1       0   264.4    .045       0   312.6      .1       0
Bank Sta=264.4,312.6
XS Rating Curve= 0 ,0
Exp/Cntr=0.3,0.1

Type RM Length L Ch R = 1 ,60264.4 ,98.2,142.9,182.2
XS GIS Cut Line= 3
     1878062.792      514438.934     1877710.362      514586.503
     1877463.834      514735.809
#Sta/Elev= 30
       0  864.68    39.2  839.31      49  834.77    58.8  833.51   186.1  832.85
   195.9  831.42   205.7  828.46   215.5  827.48   225.3   827.4   235.1  827.42
   264.5  834.46   303.7  838.72   313.5  841.67   323.3  847.33   352.7  867.22
   382.1  885.84   401.3  896.49   420.5  905.38   449.3   916.3   458.9   919.4
   478.2   924.3   487.8   928.1   497.4  932.94   526.2  949.29   545.4  959.07
   564.6  967.12   583.8  974.34     603  980.81   622.3  986.31   670.3   996.1
#Mann= 3 , 0 , 0
       0      .1       0   205.7    .045       0   235.1      .1       0
Bank Sta=205.7,235.1
XS Rating Curve= 0 ,0
Exp/Cntr=0.3,0.1

Type RM Length L Ch R = 1 ,60121.5 ,122.9,116.1,114.6
XS GIS Cut Line= 3
     1878007.237      514367.753     1877837.098      514431.989
     1877663.487      514301.781
#Sta/Elev= 29
       0  862.17    19.1  850.24    38.3  838.58    47.9  833.69    57.4  831.79
    86.1  831.51   124.4  831.45   143.6  831.21   172.3   831.2   191.3   829.8
   200.7  829.03   210.2  828.01   219.6  827.37     229  827.08   238.5   826.9
   266.8  826.91   285.6  827.95   295.1  829.26   304.5  831.27     314  834.04
   323.4  837.46   332.8  841.46   342.3  845.19   351.7  848.36   361.1  850.72
   370.6  852.66     380  854.43   389.4  856.46   398.9  858.66
#Mann= 3 , 0 , 0
       0      .1       0   219.6    .045       0   266.8      .1       0
Bank Sta=219.6,266.8
XS Rating Curve= 0 ,0
Skew Angle= 55
Exp/Cntr=0.3,0.1

Type RM Length L Ch R = 1 ,60005.4 ,239.5,200.9,162.4
XS GIS Cut Line= 4
     1878015.917      514300.045     1877845.779      514364.281
     1877649.795      514222.309      1877581.89      514242.753
#Sta/Elev= 28
       0  884.82    38.3  863.04    76.6  840.85    86.1  835.44    95.7  832.45
   105.3  831.83   124.4  831.56   230.3  831.36   239.9  830.87   249.6  830.17
   259.3  829.39   278.7   827.5   288.3  827.13   297.9   826.9   336.7   826.9
   356.1  827.42   365.8  828.78   375.5  829.95   385.1  831.25   404.5  833.61
   414.2  835.02   423.9  836.98   432.7  842.71   441.6  848.91   468.2   868.1
     477  873.88   485.9  879.22   494.8  884.24
#Mann= 3 , 0 , 0
       0      .1       0   278.7    .045       0   356.1      .1       0
Bank Sta=278.7,356.1
XS Rating Curve= 0 ,0
Skew Angle= 55
Exp/Cntr=0.3,0.1

Type RM Length L Ch R = 1 ,59804.4 ,151.5,157.1,162.6
XS GIS Cut Line= 2
     1877899.598      514001.434     1877545.431      514162.892
#Sta/Elev= 29
       0  894.44     9.7  887.37    48.6  859.33    58.4  852.34    77.8  838.26
    87.6  832.72    97.3   830.2     107  830.02   126.5  830.28   155.7  830.46
   194.6   830.5   204.4   830.4   214.1  829.59   223.8  827.46   233.5  826.59
   243.3  826.35   262.7  826.56   272.5  828.23   282.2  830.55   291.9  831.62
   311.4  831.92   321.1  832.27   330.8  835.37   340.6  841.81   350.3     849
     360     856   369.8   862.6   379.5  868.87   389.2  874.82
#Mann= 3 , 0 , 0
       0      .1       0   223.8    .045       0   262.7      .1       0
Bank Sta=223.8,262.7
XS Rating Curve= 0 ,0
Exp/Cntr=0.3,0.1

Type RM Length L Ch R = 1 ,59647.4 ,470.2,454.8,439.4
XS GIS Cut Line= 4
     1877950.548      513841.785     1877818.169      513918.825
     1877558.838      513966.568     1877419.949      514057.714
#Sta/Elev= 30
       0  965.03     9.6  960.48    86.2  926.73    95.7  922.12   105.3  915.78
   114.9  907.17   124.4   897.3     134  886.78   153.2  864.99   162.9   855.4
   172.7  846.14   182.5  837.74   192.2  831.89     202  829.73   260.6  829.61
   280.1   828.5   299.7  826.22   319.2  825.81     329   826.4   338.7  828.02
   348.5  830.32   358.3  831.21   455.9  831.11   475.5  831.56   485.3  834.62
     495  840.83   534.1  869.12   553.7  882.66   563.4  888.22     583  895.37
#Mann= 3 , 0 , 0
       0      .1       0   299.7    .045       0     329      .1       0
Bank Sta=299.7,329
XS Rating Curve= 0 ,0
Exp/Cntr=0.3,0.1

Type RM Length L Ch R = 1 ,59192.6 ,295.6,299,302.4
XS GIS Cut Line= 2
     1877583.772      513386.984      1877151.48      513878.304
#Sta/Elev= 30
       0 1006.74     9.8 1004.89    19.5 1002.11    29.3  998.07    39.1  993.08
    68.4  977.66    97.7  961.74     166  923.85   195.4  907.96   205.1  902.21
   214.9  894.99   234.4   877.9   283.3   833.6     293  826.13   302.8  822.88
   312.6  822.38   332.1  822.02   351.6   821.7   364.8822.1436   380.9  822.66
   400.5  826.91   410.2  828.29   478.6  833.18   488.4  835.55   498.1  840.14
   507.9  845.81     586   893.4   595.8  899.06   634.9  920.08   654.4  930.98
#Mann= 3 , 0 , 0
       0      .1       0   332.1    .045       0   364.8      .1       0
Bank Sta=332.1,364.8
XS Rating Curve= 0 ,0
Exp/Cntr=0.3,0.1

Type RM Length L Ch R = 1 ,58893.5 ,268.4,258.6,248.8
XS GIS Cut Line= 3
     1877340.716      513284.554     1877042.105       513536.29
      1876995.23      513616.151
#Sta/Elev= 30
       0  949.19    19.5  940.52    48.8  929.04    68.4  920.57    87.9  911.48
   107.4  901.24   126.9  890.38   136.7  883.76   146.5  875.96   156.2  867.03
   175.8  847.04   185.5  838.01   195.3  830.24     205  824.64   214.8  822.69
   253.9  820.44   263.6   820.3   283.2  820.34   292.9  820.72   302.7   823.2
   312.4   826.4   322.2  828.65     332  829.35   409.1  831.06   418.3  831.49
   427.6  833.33   436.9  837.23   446.1  842.53   455.4  847.98   483.2  865.69
#Mann= 3 , 0 , 0
       0      .1       0   253.9    .045       0   292.9      .1       0
Bank Sta=253.9,292.9
XS Rating Curve= 0 ,0
Exp/Cntr=0.3,0.1

Type RM Length L Ch R = 1 ,58634.9 ,254.8,206.9,158.1
XS GIS Cut Line= 3
     1877004.055      513129.678     1876890.123      513373.819
     1876860.826      513557.196
#Sta/Elev= 30
       0  924.31    38.5   899.9    48.1  893.38    57.7  885.45      77  866.57
    86.6  856.05    96.2   844.7   105.8  834.01   115.5  826.42   125.1  823.36
   134.7  822.86     154  822.64   163.6  822.23   173.2  821.28   182.8  820.32
   192.4   820.2   202.1   820.2   211.7  821.49   230.9  826.92   240.6  828.27
   259.8   828.8     289  828.26   337.8  828.94   357.4  830.14   376.9  832.75
   386.7  835.14   396.5  839.11   435.6  860.04   445.3  864.65   455.1  868.45
#Mann= 3 , 0 , 0
       0      .1       0   173.2    .045       0   211.7      .1       0
Bank Sta=173.2,211.7
XS Rating Curve= 0 ,0
Exp/Cntr=0.3,0.1

Type RM Length L Ch R = 1 ,58428   ,160.1,178.6,197.1
XS GIS Cut Line= 5
     1876732.858      513024.132     1876704.744      513060.877
     1876770.384      513197.804     1876822.467      513381.832
     1876810.315      513523.325
#Sta/Elev= 30
       0  865.76     9.2  861.11    18.5     856    27.8  850.36      37  844.45
    46.3   837.9    84.2  827.55    93.7  825.32   103.2  823.41   112.7  821.82
   122.2  820.54   131.7  819.81   150.7  819.47   179.1  819.59   198.1  819.96
   207.7  820.52   217.2  821.47   255.5  826.57     265  827.49   274.6  828.05
   312.9  827.71   370.2  828.06   389.4  827.94   427.2  829.53   436.7  829.62
   455.6  828.87     484  829.57     503   831.1   521.9  834.67   531.4  837.17
#Mann= 3 , 0 , 0
       0      .1       0   131.7    .045       0   198.1      .1       0
Bank Sta=131.7,198.1
XS Rating Curve= 0 ,0
Skew Angle= 45
Exp/Cntr=0.3,0.1

Type RM Length L Ch R = 1 ,58249.5 ,170.8,225,279.7
XS GIS Cut Line= 5
     1876669.768      512961.515     1876578.418      513008.688
     1876679.969      513216.156     1876732.053      513400.184
       1876719.9      513541.677
#Sta/Elev= 30
       0  841.77    18.7   831.5      28  827.85    37.4   826.4    46.7  825.98
    65.4  825.48   112.4  824.55   122.1  823.98   131.7   822.7   141.3  820.88
   150.9  819.65   160.6  819.11   179.8   819.2   193.3  819.82   237.6  822.51
   266.4  823.44   314.6  825.71   343.4  826.52   400.7  827.32   419.9  827.78
   467.7  829.81   486.8  830.84   496.4   830.9   505.9  831.24   525.1  832.23
   591.3  836.98   600.8  837.49   619.7  838.06   629.2  838.19   667.1  838.13
#Mann= 3 , 0 , 0
       0      .1       0   150.9    .045       0   193.3      .1       0
Bank Sta=150.9,193.3
XS Rating Curve= 0 ,0
Skew Angle= 45
Exp/Cntr=0.3,0.1

Type RM Length L Ch R = 1 ,58024.4 ,163.9,162.6,161.3
XS GIS Cut Line= 3
     1876661.165      512934.557     1876396.506      512946.994
     1876194.683      512986.057
#Sta/Elev= 29
       0  840.76     9.8  835.42    19.6  830.35    29.4   827.1    39.2  826.11
    68.7  825.09    98.1  823.89     157  821.83   166.8  821.07   176.6  819.79
   182.7819.0948   186.4  818.67   196.3  818.39   206.1   818.4   215.9     820
   225.7  826.18   235.5  834.39   245.3  841.73   255.1  848.85   274.7  863.33
   284.5  870.44   294.3  877.43   313.9  891.03   333.5  904.28     353  917.08
   372.6  929.28   411.8  953.16   441.2  970.71   470.5  988.44
#Mann= 3 , 0 , 0
       0      .1       0   182.7    .045       0   215.9      .1       0
Bank Sta=182.7,215.9
XS Rating Curve= 0 ,0
Exp/Cntr=0.3,0.1

Type RM Length L Ch R = 1 ,57861.9 ,151.8,170.3,189.5
XS GIS Cut Line= 2
     1876640.557       512764.01     1876389.906      512790.052
#Sta/Elev= 29
       0  852.06     9.7  846.78    19.4  841.45    29.1  836.17    38.8  830.93
    48.5  826.68    58.2     825    67.8     825    77.5  825.01    87.2  825.08
    96.9   825.1   106.6  825.19   116.3  825.11     126  825.02   135.7  823.83
   145.4   821.5   155.1   819.3   162.6  818.51   164.8  818.28   174.5  818.26
   177.6  818.27   184.2  818.28   193.8  818.03   203.5   822.9   213.2  830.89
   222.9  838.31   232.6  844.65   242.3  850.87     252  856.98
#Mann= 3 , 0 , 0
       0      .1       0   155.1    .045       0   203.5      .1       0
#XS Ineff= 2 , 0
          110.57  827.12
Permanent Ineff=
       F       F
Bank Sta=155.1,203.5
XS Rating Curve= 0 ,0
Exp/Cntr=0.3,0.1

Type RM Length L Ch R = 1 ,57691.6 ,83.8,81.9,79.1
XS GIS Cut Line= 2
     1876647.495      512745.566     1876332.087      512525.769
#Sta/Elev= 27
       0  858.72    28.8  848.91    86.5  828.79    96.1  826.25   105.7  824.35
   115.3  823.05   134.6   822.3   153.8  821.68   182.6  821.16   192.2  820.51
   201.8   819.3   211.4  817.76     221  816.61   240.3  816.46   249.9   817.1
   259.5  818.38   269.1  820.16   278.7  822.07   288.3  823.53   307.6  826.87
   317.2  828.65   326.8  830.81   336.4  833.08     346  835.69   355.6   838.6
   365.2  841.74   384.4  848.56
#Mann= 3 , 0 , 0
       0      .1       0   211.4    .045       0   249.9      .1       0
Bank Sta=211.4,249.9
XS Rating Curve= 0 ,0
Skew Angle= 30
Exp/Cntr=0.3,0.1

Type RM Length L Ch R = 1 ,57609.7 ,238.3,214.5,190.8
XS GIS Cut Line= 2
      1876648.86      512667.845     1876333.452      512448.049
#Sta/Elev= 30
       0  871.69    28.8   861.8    57.7  851.52    76.9  844.22   105.7  832.78
   124.9  825.04   134.6  822.59   144.2  821.41   153.8  821.08   182.6  821.13
   192.2  820.86   201.8  820.06   211.4   818.7  216.42817.8843     221  817.14
   230.7  816.61   240.3  816.48   249.9  817.03   259.5  818.42   269.1  820.83
   278.7   822.4   288.3  823.39   297.9  824.14   307.6  824.75   336.4  825.32
     346  825.76   355.6  826.43   365.2  828.14   374.8  830.79   384.4  833.74
#Mann= 3 , 0 , 0
       0      .1       0  216.42    .045       0   249.9      .1       0
Bank Sta=216.42,249.9
XS Rating Curve= 0 ,0
Skew Angle= 30
Exp/Cntr=0.3,0.1

Type RM Length L Ch R = 1 ,57395.2 ,199.6,136.4,82.5
XS GIS Cut Line= 2
     1876614.515      512248.602     1876324.802      512379.895
#Sta/Elev= 28
       0  883.78     9.6  880.36    28.9  873.84    38.6  870.82    48.2  867.94
    67.5  862.67    77.1  858.98    86.8   853.7    96.4   847.9     106   841.8
   115.7  835.36   125.3  829.19   134.9  823.98   144.6  820.14   154.2  817.61
   163.9  816.61   173.5  816.29   183.1  816.59   184.8816.8267   192.8  817.94
   202.4  819.74     212  820.99   221.7  821.61   250.6  822.54   260.2  822.94
   298.8  824.27   308.4   825.6   318.1  829.06
#Mann= 3 , 0 , 0
       0      .1       0   154.2    .045       0   184.8      .1       0
Bank Sta=154.2,184.8
XS Rating Curve= 0 ,0
Exp/Cntr=0.3,0.1

Type RM Length L Ch R = 1 ,57258.7 ,167.3,193.2,209.6
XS GIS Cut Line= 4
     1876386.203      511880.781      1876338.24      512009.742
     1876393.325      512271.258     1876324.738      512358.862
#Sta/Elev= 30
       0  858.66     9.8  856.72    19.7  853.92    39.3   845.7    49.1  841.82
    68.8  834.32    78.6  830.96    88.4   828.1    98.3  825.88   108.1  824.13
   117.9  823.37   137.6  822.66     233  820.86   242.6  820.41   280.8  816.78
   290.3  816.03   299.8  815.56   318.9  815.97   328.5  816.02   347.1  816.22
   357.1  816.58   366.7  816.69   376.2  817.42   385.8  818.47   404.8  820.02
   414.1  820.94   451.2  822.22   497.6  824.06   506.8  824.84   516.1  827.03
#Mann= 3 , 0 , 0
       0      .1       0   290.3    .045       0   328.5      .1       0
Bank Sta=290.3,328.5
XS Rating Curve= 0 ,0
Skew Angle= 50
Exp/Cntr=0.3,0.1

Type RM Length L Ch R = 1 ,57065.5 ,241.4,271.8,302
XS GIS Cut Line= 4
     1876276.305       511837.92     1876230.714      511961.118
     1876285.624      512221.804     1876217.038      512309.407
#Sta/Elev= 30
       0  823.56    28.2  822.96   103.2  820.99   131.4  820.58   150.4  820.58
   178.9   820.3   188.4  819.46     198  817.77   207.5   815.7     217  814.06
   226.5  813.54     236  813.58     255  814.35   264.6  815.15   274.1  816.52
   283.6   817.7   293.1  818.27   350.2  820.35   359.7  820.59   369.2  821.17
   388.2  823.34   397.8  824.27     407  827.95   434.9  840.11   453.4  848.73
   462.7   853.3   471.9   858.1   490.5  868.72   499.8  873.93     509  878.89
#Mann= 3 , 0 , 0
       0      .1       0     217    .045       0     255      .1       0
Bank Sta=217,255
XS Rating Curve= 0 ,0
Skew Angle= 50
Exp/Cntr=0.3,0.1

Type RM Length L Ch R = 1 ,56793.7 ,215,230.4,247.2
XS GIS Cut Line= 2
     1876200.846      511749.765     1876009.575      511924.323
#Sta/Elev= 30
       0  822.11     9.6  821.95    19.2  821.82    28.8  821.69    38.4  821.61
      48  821.59    57.5  821.52    67.1   821.5    76.7  821.43    86.3  821.32
    95.9  821.16   105.5  821.03   115.1   820.3   124.7   817.5   134.3  813.68
   139.2  813.36   143.9  813.06   153.4     813   154.2     813     163  813.04
   172.6  814.64   182.2  818.61   191.8  825.28   201.4  833.35     211  841.55
   220.6  849.94   230.2  858.54   239.8  867.17   249.4  875.73     259  884.06
#Mann= 3 , 0 , 0
       0      .1       0   134.3    .045       0     163      .1       0
Bank Sta=134.3,163
XS Rating Curve= 0 ,0
Exp/Cntr=0.3,0.1

Type RM Length L Ch R = 1 ,56563.2 ,90.4,91,90.3
XS GIS Cut Line= 6
     1876549.411      511607.326     1876288.995      511700.642
     1876172.817      511704.314      1875980.06      511669.611
     1875846.726      511680.028     1875784.437      511728.854
#Sta/Elev= 30
       0  852.85    28.6  837.29    38.2  832.64    47.7  829.35    57.2  828.01
   104.9  826.77   162.2  824.11   190.8  823.24   209.9  823.14     248  824.72
   276.6  825.03     296  824.66   354.1  822.42   412.4  822.11     530  817.02
   549.6  816.43   578.9  816.37   588.7  815.66   607.8  812.06   626.9  811.44
   636.5  812.41   655.6  816.28   665.2   817.3   722.5  820.42   731.3  822.61
     740   826.3   757.6  835.59   766.4  839.38   775.2  842.02   801.6  845.53
#Mann= 3 , 0 , 0
       0      .1       0   607.8    .045       0   636.5      .1       0
Bank Sta=607.8,636.5
XS Rating Curve= 0 ,0
Exp/Cntr=0.3,0.1

Type RM Length L Ch R = 1 ,56472.2 ,232.9,200.3,167.7
XS GIS Cut Line= 6
     1876260.783      511306.762     1876206.461      511474.897
     1876112.118       511602.05     1875836.726      511602.319
     1875763.859      511654.503     1875769.912      511722.524
#Sta/Elev= 30
       0   945.6    19.6   944.3    49.1  939.82    68.7  935.83    88.4  930.05
    98.2  928.02   147.2  921.91   157.1  920.08   166.9  916.87   195.3  903.65
   232.6  883.84   269.8  859.81   288.5  845.94   307.1  831.37   316.4  825.51
   325.7  822.58   382.5  818.98   458.4   815.9   496.6  812.82   525.2  811.47
   544.3  811.28   553.9  811.28   563.4  812.14   582.5  817.56   592.1  818.04
     665  817.71   720.3   820.6   730.1  822.69   749.6  830.81   769.1  839.77
#Mann= 3 , 0 , 0
       0      .1       0   525.2    .045       0   563.4      .1       0
Bank Sta=525.2,563.4
XS Rating Curve= 0 ,0
Exp/Cntr=0.3,0.1

Type RM Length L Ch R = 1 ,56271.9 ,273.9,246.9,219.6
XS GIS Cut Line= 3
     1875783.801      511294.572     1875743.871       511661.76
     1875751.683      511723.392
#Sta/Elev= 29
       0   903.6    19.4   893.4    29.2  888.41    38.9  883.19    48.6   877.2
    97.2  843.69   116.6   830.5   136.1  817.41   145.8  812.31   155.5  810.52
   165.2   810.6   168.3811.1475     175  812.32   184.7  815.58   194.4  817.44
   262.4  816.71   291.6     817   301.3     817     311   816.8   320.8  816.72
   330.5  817.18   340.2  817.75   359.6  819.05   378.2  820.11   387.1  820.52
     396  821.62   404.8  824.23   413.7     828   431.5  836.18
#Mann= 3 , 0 , 0
       0      .1       0   145.8    .045       0   168.3      .1       0
Bank Sta=145.8,168.3
XS Rating Curve= 0 ,0
Exp/Cntr=0.3,0.1

Type RM Length L Ch R = 1 ,56025   ,329.4,327.5,325.6
XS GIS Cut Line= 4
     1875427.378      511457.574     1875520.703      511542.616
     1875606.297      511587.897     1875705.144       511755.22
#Sta/Elev= 29
       0  925.66     9.7  919.05    38.8  896.76    77.7  867.21    87.4  860.03
    97.1  853.19   106.8  846.55   135.9  827.68   155.3  815.63     165  811.19
   165.7811.0653   174.7  809.46   184.4  809.51   185.7809.7321     194  811.15
   203.7  814.98   213.4  817.18   223.1  817.38   271.7  816.54   291.1  816.42
   300.8  816.48   310.6  816.64   320.3  816.91   339.7  817.64   378.6  819.77
   388.3  820.82     398  823.86   407.7  828.36   417.4  833.28
#Mann= 3 , 0 , 0
       0      .1       0   165.7    .045       0   185.7      .1       0
Bank Sta=165.7,185.7
XS Rating Curve= 0 ,0
Exp/Cntr=0.3,0.1

Type RM Length L Ch R = 1 ,55697.4 ,516.6,552.2,587.7
XS GIS Cut Line= 4
     1875282.864      511752.896     1875343.791      511827.133
     1875569.316      511923.428     1875708.754      512063.969
#Sta/Elev= 30
       0  873.08    28.8  861.24    38.4  856.66    67.2  841.08    86.4  831.62
      96  827.21   125.5   815.3   135.3  812.69   145.1  811.69   174.5  810.15
   184.3  809.39   194.1  808.28   203.9  807.14   213.7  807.46   223.6   808.9
   233.4  811.96   243.2   813.5     253  813.92     302  814.65   311.8  815.06
   321.6  816.91   331.4  821.24   350.7  831.69   388.4  851.48   407.2  861.76
   416.7  867.12   435.5  878.33   463.8  896.28   473.2  901.75   539.2  938.26
#Mann= 3 , 0 , 0
       0      .1       0   194.1    .045       0   223.6      .1       0
Bank Sta=194.1,223.6
XS Rating Curve= 0 ,0
Exp/Cntr=0.3,0.1

Type RM Length L Ch R = 1 ,55145.3 ,259.7,262.8,265.9
XS GIS Cut Line= 3
     1875110.609      511746.215     1874987.996      512040.269
     1874935.913      512269.218
#Sta/Elev= 30
       0  849.51    48.3  831.15    77.2  819.04    86.9   816.3    96.5  815.35
   135.2   814.8   173.8  814.58   202.7  814.04   212.4   812.8     222  809.45
   231.7  805.38   241.4  804.13   260.7   804.2   266.7806.8706   270.3  808.47
     280  818.48   289.6  828.76   299.3  837.03   308.9  843.99   318.6  850.52
   347.9  869.14   367.5  881.02   377.3   886.7   387.1  891.95   396.9  896.65
   445.8  918.53   494.7  937.93   514.3  946.02   533.8  955.18   553.4  965.26
#Mann= 3 , 0 , 0
       0      .1       0   231.7    .045       0   266.7      .1       0
Bank Sta=231.7,266.7
XS Rating Curve= 0 ,0
Exp/Cntr=0.3,0.1

Type RM Length L Ch R = 1 ,54882.5 ,428.3,429.6,430.9
XS GIS Cut Line= 2
     1874944.593      511581.284      1874736.26      511933.932
#Sta/Elev= 30
       0  895.19    19.5  883.45      39  872.02    58.5  861.12    68.3  855.93
    97.5  841.07     117  830.62   126.8  825.85   136.5  821.54   146.3  817.89
     156  815.06   165.8  813.28   175.5  812.65   224.3  811.19   243.8  810.42
   263.3  809.28   273.1   807.8   282.8  804.48   292.6  801.56   302.3  801.01
   321.8  801.12   331.6   805.6   341.3  816.72   351.1  828.26   360.8  837.09
   370.6  843.27   380.3  847.76   390.1  851.77   399.8  856.39   409.6  861.84
#Mann= 3 , 0 , 0
       0      .1       0   292.6    .045       0   321.8      .1       0
Bank Sta=292.6,321.8
XS Rating Curve= 0 ,0
Exp/Cntr=0.3,0.1

Type RM Length L Ch R = 1 ,54452.9 ,167.5,157.8,148.1
XS GIS Cut Line= 4
     1874849.888       511349.46     1874530.097      511461.927
     1874382.527      511681.111     1874364.081      511800.468
#Sta/Elev= 30
       0  984.04    19.4  974.38    58.1  950.03    77.5  938.92   106.5  925.51
     155  906.86   164.6  900.64     184  884.88   193.7  878.22   213.1  866.71
   232.4  856.52   251.8  847.36   300.2     830   309.9   825.2   319.6   819.3
   329.3  814.88     339  812.67   368.4  810.96   397.7  807.98     476  806.81
   495.6  801.27   505.4  800.69     525801.3194   544.5  807.44   554.3  808.54
   612.5  809.53   621.8  810.01   631.1   812.2   677.6  833.72     724  858.22
#Mann= 3 , 0 , 0
       0      .1       0   495.6    .045       0     525      .1       0
Bank Sta=495.6,525
XS Rating Curve= 0 ,0
Exp/Cntr=0.3,0.1

Type RM Length L Ch R = 1 ,54295.1 ,606.1,568.6,530.9
XS GIS Cut Line= 4
       1874184.8      511173.474      1874302.41      511464.898
     1874267.687      511674.968     1874318.035      511817.329
#Sta/Elev= 30
       0  988.33     9.8  983.04    19.6  977.14    98.2  926.72   127.7  907.28
   147.3  893.68   196.4  858.59   225.9   838.5   245.5  826.68   265.2  815.55
     275  811.74   284.8  810.49   323.9  809.95   343.3  809.09   362.6  807.66
     382  801.12   391.7   800.3   401.2  800.58   403.7801.0315     411  802.35
   420.7  805.03   430.4  806.71   469.1  808.18   564.9  810.94   574.4  812.08
   583.8  815.67   621.6  838.49     631  843.61   659.3  856.07   678.2  865.26
#Mann= 3 , 0 , 0
       0      .1       0     382    .045       0   403.7      .1       0
Bank Sta=382,403.7
XS Rating Curve= 0 ,0
Exp/Cntr=0.3,0.1

Type RM Length L Ch R = 1 ,53726.5 ,438,445.4,452.7
XS GIS Cut Line= 4
     1873700.778      511831.829     1873862.993      511873.397
     1874151.774      511894.478     1874242.866      511919.455
#Sta/Elev= 30
       0  922.18    18.6  915.25    27.9  911.15    55.8  897.33    74.4  887.74
   102.3  872.56   120.9  862.16   130.2  857.29   139.6  853.07   158.2  845.56
   167.5  840.94   177.1  835.08   186.8     828   196.4  820.18   206.1  812.85
   215.7  807.12   225.4  802.82     235  799.86   237.2799.6213   244.7   798.8
   257.2799.0195     264  799.29   273.6  800.21   292.9  803.25   399.1  807.26
   408.8  808.75   418.4  812.18   466.4   833.8   513.7  857.03   551.5  875.28
#Mann= 3 , 0 , 0
       0      .1       0   237.2    .045       0   257.2      .1       0
Bank Sta=237.2,257.2
XS Rating Curve= 0 ,0
Exp/Cntr=0.3,0.1

Type RM Length L Ch R = 1 ,53281.1 ,311.4,341.1,369.4
XS GIS Cut Line= 3
     1873723.611      512233.144     1874044.263      512367.101
     1874330.107      512449.373
#Sta/Elev= 30
       0  842.57      29  833.75    38.6  829.98    48.3  825.31    77.2  809.63
    86.9  805.24    96.5  802.92   115.8  801.98   135.1  801.73   183.4  800.32
   193.1  799.82     222  796.66   231.7  796.61     251  796.93   270.3  801.29
   279.9  804.56   289.6  808.83   308.9   818.2   318.6   822.5   328.2  826.28
   337.9  829.91   357.1  834.94   366.7   837.9   376.3   841.5   424.3  861.74
   491.4  888.17   520.2  897.95   558.6  911.65   616.2  937.66     645  949.02
#Mann= 3 , 0 , 0
       0      .1       0     222    .045       0     251      .1       0
Bank Sta=222,251
XS Rating Curve= 0 ,0
Exp/Cntr=0.3,0.1

Type RM Length L Ch R = 1 ,52940.1 ,431.7,444.9,459.8
XS GIS Cut Line= 4
      1873703.57      512248.966     1873730.994      512463.085
     1873711.332       512728.83     1873622.352       512890.27
#Sta/Elev= 30
       0  841.33    29.4  829.42    58.9  818.18    88.3  807.44    98.1  804.79
   107.9  803.87   215.9  802.88   263.4   801.8     273   801.3   282.5  800.16
     311  793.92   320.6  793.29   339.6   793.6   349.1  796.64   368.1  808.11
   377.6  812.28   387.2   815.2   444.3  828.84   482.3   839.8   501.7  847.17
   511.4  851.62   521.2  856.76   550.2  873.54     560  878.19   589.1  888.86
   598.8  893.51   618.2  904.03   637.6  915.22   647.3  921.18   666.7  933.92
#Mann= 3 , 0 , 0
       0      .1       0     311    .045       0   339.6      .1       0
Bank Sta=311,339.6
XS Rating Curve= 0 ,0
Exp/Cntr=0.3,0.1

Type RM Length L Ch R = 1 ,52495.1 ,320.7,313.5,305.7
XS GIS Cut Line= 2
     1873567.504      512194.117     1873280.604       512486.29
#Sta/Elev= 30
       0  850.31     9.8  845.19      39  829.36    58.5  819.21    68.2  814.38
      78  809.69    87.8  805.39    97.5  801.65   107.2  799.29     117  798.16
   126.7  797.32   146.2  795.78   165.7  794.44   175.5  793.94   204.7  793.14
   214.5  792.23   224.2  791.59     234  791.44   243.7   791.8   253.5  792.72
   263.2  794.63   282.7  800.18   292.5  803.16   302.2  806.34     312  809.98
   321.7  814.76   331.5  820.48   360.7  838.72     390  856.78   409.5  868.94
#Mann= 3 , 0 , 0
       0      .1       0   214.5    .045       0   253.5      .1       0
Bank Sta=214.5,253.5
XS Rating Curve= 0 ,0
Exp/Cntr=0.3,0.1

Type RM Length L Ch R = 1 ,52181.6 ,272.8,263.4,253.9
XS GIS Cut Line= 3
     1873282.231      511963.127     1873140.043      512301.089
     1873141.534      512438.681
#Sta/Elev= 30
       0  890.84     9.6  885.67      29  874.68    67.5  852.29    86.8  841.19
   106.1  830.29   115.8  824.85   173.7  793.15   183.3  790.55     193   790.1
   202.6  790.41   206.3791.1194   212.3  792.27   221.9   795.7   231.6   797.7
   241.2  797.67   260.5  796.97   289.5  796.17   299.1  796.04   308.8  796.02
   318.4  796.19   328.1   797.5   337.7  801.65   366.6  817.13   396.1  834.19
   435.4  855.96   445.3  860.92   455.1  865.13   464.9  869.04   504.3  883.77
#Mann= 3 , 0 , 0
       0      .1       0   183.3    .045       0   206.3      .1       0
Bank Sta=183.3,206.3
XS Rating Curve= 0 ,0
Exp/Cntr=0.3,0.1

Type RM Length L Ch R = 1 ,51918.3 ,363.7,341.1,318.5
XS GIS Cut Line= 4
     1873013.217      511829.034     1872955.295      512024.754
     1872956.961      512119.808     1873072.609      512456.672
#Sta/Elev= 30
       0  915.06     9.7  909.26    19.4  904.52    48.6  893.49   116.6   866.4
   126.4  861.33   136.1  855.02   184.7  821.26   204.1  808.37   232.6  792.86
   242.1  789.92   251.6  789.19   261.2  789.99     265790.9946   280.2  795.78
   289.7  797.93   299.2  798.34   337.7  796.27   405.1  794.74   462.8  794.99
   491.7  796.17   501.3  797.32     511  802.02   539.8  820.14   549.5  826.38
   578.3  846.26     588  852.37   616.8  869.15   626.5  874.34   655.3  887.69
#Mann= 3 , 0 , 0
       0      .1       0   242.1    .045       0     265      .1       0
#XS Ineff= 2 , 0
                          464.52          809.17
Permanent Ineff=
       F       F
Bank Sta=242.1,265
XS Rating Curve= 0 ,0
Exp/Cntr=0.3,0.1

Type RM Length L Ch R = 1 ,51577.2 ,381.2,359.7,338.1
XS GIS Cut Line= 3
     1872535.757      512195.483      1872882.33      512411.929
     1873035.434      512510.017
#Sta/Elev= 30
       0  932.77    77.8  884.74    97.3  873.71   136.2  852.36   155.7  841.26
   165.4  835.03   194.6  814.54   204.3  807.58     214  800.18   223.8  791.67
   231.5787.5421   233.5  786.47   243.2  785.48     253   786.8   272.4  792.36
   282.1  793.86   398.9  795.42   408.6   795.8   418.2   798.2   427.8  802.29
   456.5  816.26   475.6   826.7   504.3     843   513.9   848.1   523.4  852.83
     533  857.22   542.6   861.1   561.7  868.38   571.3  872.37   590.4  880.94
#Mann= 3 , 0 , 0
       0      .1       0   231.5    .045       0     253      .1       0
Bank Sta=231.5,253
XS Rating Curve= 0 ,0
Exp/Cntr=0.3,0.1

Type RM Length L Ch R = 1 ,51217.5 ,279.8,279.4,279
XS GIS Cut Line= 3
     1872555.984       512730.75     1872800.775       512628.32
     1873010.845      512600.542
#Sta/Elev= 30
       0  883.93    19.7   872.6    29.5  866.18    39.3  859.22      59  844.61
    88.4  821.98   108.1  807.17   127.8  793.21   137.6  787.55   147.4  784.94
   167.1  784.14   176.9  782.59   186.7  780.62   196.6  780.85   206.4  786.35
   216.2  791.01     226  792.43   255.5  794.09   265.4  794.23   284.6  793.53
   294.2   792.8   313.5   790.4   323.2  789.55   332.8  790.75   342.4   794.3
     352  798.98   361.7  804.06   400.2  825.86   438.7  845.96   477.3  865.52
#Mann= 3 , 0 , 0
       0      .1       0   167.1    .045       0   206.4      .1       0
#XS Ineff= 2 , 0
                          267.71           802.2
Permanent Ineff=
       F       F
Bank Sta=167.1,206.4
XS Rating Curve= 0 ,0
Exp/Cntr=0.3,0.1
