HEC-RAS study FALLINGRCR.prj: FALLINGRCR

--- FALLINGRCR.g01 (geometry) --- (continued)

Type RM Length L Ch R = 1 ,50938.1 ,313.3,312.7,311.9
XS GIS Cut Line= 2
      1872613.42      513013.519     1873087.595      512805.186
#Sta/Elev= 30
       0  921.48     9.8  915.21    19.5  908.87    29.3  902.65    58.6  883.69
      88  865.09   107.5  852.61     127  839.88   146.6  826.84   166.1  814.28
   175.9  808.37   185.7   802.9   195.4  797.81   224.8  783.75   230.1 782.092
   234.5  780.72   244.3   780.2   254.1  781.45   263.8  784.07   273.6  786.91
   283.4  788.27   293.2  788.46   351.8  788.29   361.6  788.35   371.3  788.72
   381.1  790.25   390.9  794.48   410.4  805.04     430  815.54   517.9  862.25
#Mann= 3 , 0 , 0
       0      .1       0   230.1    .045       0   254.1      .1       0
Bank Sta=230.1,254.1
XS Rating Curve= 0 ,0
Exp/Cntr=0.3,0.1

Type RM Length L Ch R = 1 ,50625.4 ,466.3,485.8,504.9
XS GIS Cut Line= 4
     1872728.437      513263.085     1872884.687      513238.129
     1873124.488      513124.196     1873338.246      513127.452
#Sta/Elev= 30
       0   891.6    37.2  869.37    46.5  863.26    55.8  856.36   130.3  800.03
   139.6  793.66   148.9  789.84   158.2  788.87   197.6  788.44   207.4  788.15
   217.2  786.86   236.9  781.37   239.5781.0182   246.7  780.05   256.6  780.03
   259.5780.3992   266.4  781.28   276.2  783.46   286.1  784.66   315.6  785.56
   345.1  786.88   354.9  787.52   364.7  788.42   374.6  790.41   384.4  794.68
   423.7  815.37   501.5  853.85   530.6  868.64   569.5  890.24   637.5   929.2
#Mann= 3 , 0 , 0
       0      .1       0   239.5    .045       0   259.5      .1       0
Bank Sta=239.5,259.5
XS Rating Curve= 0 ,0
Exp/Cntr=0.3,0.1

Type RM Length L Ch R = 1 ,50139.6 ,249.9,276.6,302.8
XS GIS Cut Line= 4
     1872761.849      513440.044     1872914.649      513590.013
     1873094.783      513667.595     1873490.382       513844.59
#Sta/Elev= 30
       0  840.09    19.5  825.77    48.7  801.47    58.4  793.06    68.1  786.98
    77.8  784.64   136.2  783.19   184.9  782.47   253.3   782.9   292.6  783.82
   302.4   783.3     322  779.83   331.8  778.87   341.6  778.71   351.4  778.79
   361.2  780.13     371     785   410.2  808.62   477.6  847.13   496.9  857.72
   554.7  888.92     574  899.01   612.5  917.93   631.7  926.32   641.4  929.45
     651  931.63   660.6  933.29   699.2  938.47   776.2  950.85   843.6   959.7
#Mann= 3 , 0 , 0
       0      .1       0     322    .045       0   361.2      .1       0
Bank Sta=322,361.2
XS Rating Curve= 0 ,0
Exp/Cntr=0.3,0.1

Type RM Length L Ch R = 1 ,49863   ,653.3,655.6,658.2
XS GIS Cut Line= 4
     1872737.118      513457.313     1872823.923       513655.88
     1872822.838      513926.063     1872829.349      514133.311
#Sta/Elev= 30
       0  844.29    18.8  835.02    28.3   828.7    37.7  821.61    47.1  813.14
    56.5  801.88      66  791.34    75.4  785.56    84.8  784.37   131.9  782.28
   188.4  780.52   226.4  780.44   313.2   781.5   322.9  780.78   342.2  777.97
   351.8   777.9   371.1   778.1   380.8  779.96     400  792.88   409.7  798.63
   419.4  802.84     429  805.97   448.3  810.69     458  813.64   486.9  824.59
   524.6  837.97   581.2  856.65     600  864.24   647.1  885.71   694.2  905.41
#Mann= 3 , 0 , 0
       0      .1       0   342.2    .045       0   371.1      .1       0
Bank Sta=342.2,371.1
XS Rating Curve= 0 ,0
Exp/Cntr=0.3,0.1

Type RM Length L Ch R = 1 ,49207.4 ,448.7,453.2,457.6
XS GIS Cut Line= 3
     1872396.406      513295.637     1872369.279      513541.948
     1872331.302      513696.028
#Sta/Elev= 30
       0  840.85     9.5  836.61    38.1  824.32    47.6  820.39    76.2  809.11
    85.8  804.94    95.3  800.46   104.8  795.79   123.9  786.02   133.4  782.05
     143  779.75   152.5   778.4   181.1  774.62   190.6  774.26   200.2  774.75
   209.7  774.61   219.2  774.84   238.3  778.93   247.8  779.12   266.5  779.22
   285.1   779.5   294.5  780.75   303.8  784.62   313.1  790.64   322.5  795.17
   331.8  796.56   341.2  801.81   359.8  811.64   387.8  825.85   406.5  835.21
#Mann= 3 , 0 , 0
       0      .1       0   181.1    .045       0   219.2      .1       0
Bank Sta=181.1,219.2
XS Rating Curve= 0 ,0
Exp/Cntr=0.3,0.1

Type RM Length L Ch R = 1 ,48754.2 ,422.4,396,369.4
XS GIS Cut Line= 3
     1872036.163      513117.686     1871900.529      513546.288
     1871892.934      513633.094
#Sta/Elev= 30
       0  910.88    19.6     899    29.3  892.56    58.6  872.17      88  852.05
   136.8  815.83   156.4  802.12   166.1  795.56   185.7  782.82   195.5  778.29
   205.2  776.51   224.8  775.27   283.4  775.05     303  775.26   312.7  773.84
   322.5   771.1   332.3   769.9   361.6     770   371.4  772.86   381.1  776.95
   390.9  779.18   400.7   779.3   410.5  778.81   420.2   778.9     430  780.52
   439.8  784.17   449.6     789   468.9  799.08     527  828.07   536.7  832.31
#Mann= 3 , 0 , 0
       0      .1       0   332.3    .045       0   361.6      .1       0
#XS Ineff= 2 , 0
                          392.63           786.4
Permanent Ineff=
       F       F
Bank Sta=332.3,361.6
XS Rating Curve= 0 ,0
Exp/Cntr=0.3,0.1

Type RM Length L Ch R = 1 ,48358.2 ,474.8,475.7,476.4
XS GIS Cut Line= 3
     1871430.448      513296.273     1871724.748      513553.884
     1871800.534      513696.043
#Sta/Elev= 30
       0  908.24    58.7  868.04    68.4  861.52    78.2  855.38      88  850.14
   107.6  841.46   117.3  836.55   127.1  829.64   136.9  820.77   146.7   811.5
   166.2  792.47     176  782.34   185.8  774.08   195.6  769.71   205.3  769.09
   244.4  769.11   254.2  769.49   273.8  773.91   283.6  775.16   332.4  777.08
   410.1  778.02   419.6  778.82     429  782.08   438.5  787.55   485.9  817.88
   495.4  821.06   504.8  823.68   514.3  829.47   523.8  834.92   552.2  849.53
#Mann= 3 , 0 , 0
       0      .1       0   195.6    .045       0   254.2      .1       0
Bank Sta=195.6,254.2
XS Rating Curve= 0 ,0
Exp/Cntr=0.3,0.1

Type RM Length L Ch R = 1 ,47882.5 ,372,382.9,393.8
XS GIS Cut Line= 3
     1871138.811      513582.096     1871206.027      513724.166
     1871407.388      513913.721
#Sta/Elev= 30
       0  835.15    19.6   828.7    29.5  824.55    39.3  819.66    98.2  789.65
     108  788.84   117.9  784.47   127.7  781.06   137.5  779.41   147.4  778.52
   176.2  776.53   195.3  775.07   204.8  773.96   214.4  772.18   223.9  769.81
   233.5  767.85     243  767.12   252.5   767.1   271.6  767.48   281.1  768.27
   300.2  770.39   338.4  772.81   347.9  773.62   357.4  776.27     367  781.35
   376.5  788.21   395.6  802.78   405.1  809.19   414.6  814.84   433.7  825.44
#Mann= 3 , 0 , 0
       0      .1       0   233.5    .045       0   271.6      .1       0
Bank Sta=233.5,271.6
XS Rating Curve= 0 ,0
Exp/Cntr=0.3,0.1

Type RM Length L Ch R = 1 ,47499.6 ,254.1,253.3,252.4
XS GIS Cut Line= 3
     1871000.356      513582.096     1870924.773      513879.445
     1871013.377      514134.179
#Sta/Elev= 30
       0  828.08    19.2  823.41    28.8  820.54    67.1  807.98    76.7   804.2
   105.5   791.3     115  788.09   124.6  786.56   134.2  782.96   143.8  780.91
   153.4   780.2   201.3  778.22   230.1  777.19   316.4  774.91   326.1  774.79
   364.6   774.9   374.2   774.3   383.9  771.82   393.5  768.06   403.1  765.49
   412.8  764.88   422.4  764.91     432  765.87   441.7  770.39   451.3  777.71
   460.9  784.22   489.8   802.8   547.6  839.04   566.9  850.69   576.5  855.99
#Mann= 3 , 0 , 0
       0      .1       0   403.1    .045       0     432      .1       0
Bank Sta=403.1,432
XS Rating Curve= 0 ,0
Exp/Cntr=0.3,0.1

Type RM Length L Ch R = 1 ,47246.3 ,93.6,102.3,111.1
XS GIS Cut Line= 3
     1870578.481      513683.658     1870633.009       513839.46
      1870784.21      514225.325
#Sta/Elev= 30
       0  884.45     9.7  880.77    29.1  872.23    38.8  871.47    77.7  851.52
    97.1  842.04   135.9  825.02   174.7   810.3     194  800.79   222.9  784.98
   232.5  781.22   242.2   779.6   261.4  778.49   367.5  774.03   377.1  771.91
   386.7  767.34   396.4  764.41   425.3  763.83   434.9  763.85   444.6  764.62
   454.2  767.58   463.8  771.41   483.1  776.79   492.8  780.21   502.4  784.16
     541  803.52   550.6  807.78   560.2  810.75   569.9  811.54   579.5   810.7
#Mann= 3 , 0 , 0
       0      .1       0   396.4    .045       0   444.6      .1       0
Bank Sta=396.4,444.6
XS Rating Curve= 0 ,0
Exp/Cntr=0.3,0.1

Type RM Length L Ch R = 1 ,47144   ,56.1,56.1,56.1
XS GIS Cut Line= 3
     1870554.946      513749.395      1870629.33      513970.749
      1870629.33       514240.95
#Sta/Elev= 30
       0  863.82     9.7  859.45    48.6  842.21    68.1   833.7   116.8  812.64
   126.5  807.87   155.7  792.44   165.4  787.15   175.1   782.1   184.9   779.3
   194.6  778.36   233.5  776.22   272.1  773.57   281.8  773.01   291.4  772.59
   320.4  772.08     330  771.15   339.7  768.45   349.3  765.19     359  763.72
   368.6  763.34   387.9   762.8   397.6  763.04   407.2  765.04   416.9  768.71
   426.5  770.84   465.1   772.8   484.4  773.68   494.1  774.07   503.7  774.28
#Mann= 3 , 0 , 0
       0      .1       0   349.3    .045       0   407.2      .1       0
Bank Sta=349.3,407.2
XS Rating Curve= 0 ,0
Exp/Cntr=0.3,0.1

Type RM Length L Ch R = 1 ,47087.9 ,261.2,234.5,207.5
XS GIS Cut Line= 4
     1869940.362      513544.968     1870467.706      513647.833
     1870576.553      513981.835     1870576.553      514256.575
#Sta/Elev= 30
       0   972.5    29.3  973.86    97.7  974.47   107.5  974.03     127  970.63
   136.8  969.78   205.1  966.45     254  962.12   332.1  951.16   537.3  916.56
   566.6  905.35   595.8  889.87   605.6  886.15   615.4  884.85   664.1  859.85
   712.9  838.42   771.5  813.91     791  804.07     830  781.78   839.8  778.09
   908.2  772.31   986.7  769.76   996.5  768.97    1026763.0941  1045.6  762.31
  1055.4   762.7    1075  767.96  1084.8  769.58  1124.1  771.09  1163.3  771.45
#Mann= 3 , 0 , 0
       0      .1       0    1026    .045       0  1055.4      .1       0
Bank Sta=1026,1055.4
XS Rating Curve= 0 ,0
Exp/Cntr=0.3,0.1

Type RM Length L Ch R = 1 ,46853.4 ,522.4,498,473.5
XS GIS Cut Line= 4
     1869862.335      514151.106     1870277.774      514169.124
     1870566.762      514291.731     1870691.762      514286.523
#Sta/Elev= 30
       0  867.99    38.7  867.17      58  866.48   106.4  864.26   125.7  863.04
   135.4  862.16   154.7     860   203.1  853.86   222.4  851.75   232.1   850.9
   261.1  848.98   319.1  844.54   328.8  842.98   338.5  839.74   348.1  835.05
   377.2  819.91   415.8  798.69   464.9  776.17   474.7  771.52   484.5  765.89
   494.3  761.63   504.1  760.21   513.9  760.32   523.7  760.74   592.4  765.43
   602.2  765.89   806.7  773.98   816.4  774.96     826  776.47   854.9  781.99
#Mann= 3 , 0 , 0
       0      .1       0   494.3    .045       0   523.7      .1       0
Bank Sta=494.3,523.7
XS Rating Curve= 0 ,0
Exp/Cntr=0.3,0.1

Type RM Length L Ch R = 1 ,46355.3 ,343.5,393,441.9
XS GIS Cut Line= 3
     1870562.856      514652.408     1870686.554      514554.752
      1871096.71      514407.617
#Sta/Elev= 30
       0  777.09     9.3   780.4    18.5  781.28    27.8  777.73    37.1  769.48
    46.4  761.59    55.6  759.14    64.9  758.82    83.4  759.04    92.7  760.78
     102  764.33   111.2  766.54   120.5  767.28   139.1  767.72   167.3  769.98
     206  771.98   293.2  774.62   331.9  776.28   370.6  778.66   380.3  779.82
     390  781.72     419  787.75   438.4  792.18   457.8  797.51   467.5  800.73
   477.2  804.52   496.5  812.72   506.2  817.15   544.9  836.88   593.4  859.94
#Mann= 3 , 0 , 0
       0      .1       0    46.4    .045       0    92.7      .1       0
Bank Sta=46.4,92.7
XS Rating Curve= 0 ,0
Exp/Cntr=0.3,0.1

Type RM Length L Ch R = 1 ,45962.4 ,213.4,216.6,220
XS GIS Cut Line= 4
       1870527.7      514639.387     1870548.533      514932.356
     1870667.022      515086.002     1871130.564       515140.69
#Sta/Elev= 30
       0  780.08     9.8  776.01    19.6  772.96    29.4  771.48    97.9  771.36
   107.7  770.86   117.5   767.6   127.3  761.68   137.1  757.74   176.2  757.38
   195.8   757.1   225.2  757.92   244.8  762.41   254.6  765.44   264.3  769.98
   332.5   813.7     381  846.14   410.1  864.48   439.2  880.83   487.7  904.71
   516.9  908.02   565.5  917.36   662.8  932.48   701.7  939.73   740.6   948.5
   828.1  971.99   847.5  977.89   876.7  988.16   915.6 1003.09   954.5 1019.37
#Mann= 3 , 0 , 0
       0      .1       0   176.2    .045       0   225.2      .1       0
Bank Sta=176.2,225.2
XS Rating Curve= 0 ,0
Exp/Cntr=0.3,0.1

Type RM Length L Ch R = 1 ,45745.8 ,367.3,342.6,317.8
XS GIS Cut Line= 3
     1870256.866      514467.512     1870332.048      514743.786
     1870317.173      514946.136
#Sta/Elev= 30
       0  862.68     9.5  857.11    28.6  845.74    76.4  819.01   114.5  797.59
   133.6     787   143.2  781.76   162.2  771.69   171.8  768.75   181.3  767.98
   200.4  767.48   238.6  766.66   257.7  766.41   276.8   766.3     296  766.42
   305.6  766.39   315.3  765.73     325  763.58   344.3  757.42     354  756.68
   363.6  756.79   373.3  756.64   382.9  756.83   392.6   757.6   402.3   761.9
   440.9  784.19   450.6  789.89   469.9  801.59   479.6  806.11   489.2  807.73
#Mann= 3 , 0 , 0
       0      .1       0   344.3    .045       0   392.6      .1       0
Bank Sta=344.3,392.6
XS Rating Curve= 0 ,0
Exp/Cntr=0.3,0.1

Type RM Length L Ch R = 1 ,45403.1 ,280.4,257.4,234.2
XS GIS Cut Line= 3
     1869785.512       514703.19     1870160.512       514934.96
     1870276.397      514971.419
#Sta/Elev= 30
       0  920.65    78.4  873.03    88.2  865.78      98  856.56   107.8  846.26
   117.6   835.2     147  800.48   156.7  789.85   166.5   780.7   176.3  772.91
   186.1  766.66   195.9  761.76   205.7  758.28   225.3  754.39   235.1  753.33
   264.5  752.75   274.3   753.4   284.1  754.92   313.5  761.51   323.3  763.26
   333.1  764.22   342.9   764.6   372.3  763.94   391.9  764.28   468.9  768.56
   506.3     770   515.6  771.22     525  774.07   534.3  778.04   562.3  791.14
#Mann= 3 , 0 , 0
       0      .1       0   235.1    .045       0   274.3      .1       0
Bank Sta=235.1,274.3
XS Rating Curve= 0 ,0
Exp/Cntr=0.3,0.1

Type RM Length L Ch R = 1 ,45145.7 ,591.9,598.8,605.4
XS GIS Cut Line= 3
     1869880.564      515160.221     1870150.095      515026.106
     1870359.731       514997.46
#Sta/Elev= 30
       0  868.79    38.8   847.4    48.6  841.54    58.3  835.09    77.7  821.34
   126.2  785.32   155.4   764.4   165.1  757.63   174.8  753.38   184.5  752.21
   203.9  752.78   213.4  752.89   223.4  753.36   233.1  755.73   242.8  760.33
   252.5   763.4   262.2  764.27     301  765.84   320.3  766.26   349.1   767.2
   387.6  767.86   397.2  768.26   406.8  771.24   416.5  777.02   435.7  789.68
   445.3  795.62   454.9  800.37   464.6  804.21   493.4  814.96   512.6  822.34
#Mann= 3 , 0 , 0
       0      .1       0   174.8    .045       0   223.4      .1       0
Bank Sta=174.8,223.4
XS Rating Curve= 0 ,0
Exp/Cntr=0.3,0.1

Type RM Length L Ch R = 1 ,44546.9 ,308.5,312.9,317.2
XS GIS Cut Line= 2
     1870018.083      515621.035     1870587.536      515522.686
#Sta/Elev= 30
       0  792.28    58.8  777.19    88.2  769.18      98  766.68   107.7  764.67
   117.5   763.5   127.3  763.08   195.9  761.91   215.5  761.19   225.3  759.76
   244.9  755.23   264.5  751.82   274.2  751.02     284  750.94   303.6  751.23
   313.4  752.13   323.2  756.14     333  763.25   362.4  785.78   372.2  792.39
     382  796.86   401.6  804.43   421.2   813.3   450.6  828.48   499.5  854.77
   519.1  865.85   528.9  870.84   538.7  874.39   548.5  876.81   577.9  882.81
#Mann= 3 , 0 , 0
       0      .1       0   264.5    .045       0   313.4      .1       0
Bank Sta=264.5,313.4
XS Rating Curve= 0 ,0
Exp/Cntr=0.3,0.1

Type RM Length L Ch R = 1 ,44234   ,456,459.3,462.4
XS GIS Cut Line= 3
     1869945.232        515853.4     1870158.928      515880.112
     1870566.895      515888.611
#Sta/Elev= 30
       0  808.09    29.4  798.08    58.7  786.25    68.5  782.82    97.9  775.11
     137  766.93   156.6  764.48   176.2  762.83   195.8  762.04   225.1  762.06
   254.2  761.39     332  756.46   341.7  755.25   361.1   750.5   370.8  750.22
   380.5  750.69     400  750.53   409.7  756.01   419.4  766.53   438.8  785.13
   448.5  793.44   458.2  800.82   506.8  833.22   516.5  839.11   526.3  844.29
   555.4  856.85   565.1  859.88   574.8  860.78   584.6  860.37   623.4  857.06
#Mann= 3 , 0 , 0
       0      .1       0   361.1    .045       0     400      .1       0
Bank Sta=361.1,400
XS Rating Curve= 0 ,0
Exp/Cntr=0.3,0.1

Type RM Length L Ch R = 1 ,43774.8 ,340.1,343.7,347.4
XS GIS Cut Line= 2
     1869967.872      516289.958     1870500.164      516377.458
#Sta/Elev= 30
       0  795.47    29.4  778.32    39.2   772.8      49  768.53    58.8  765.93
    78.5  761.75    88.3  760.22    98.1  759.55   147.1  758.49   235.4  757.42
   245.2   757.2     255  756.62   264.8  754.54   274.6     751   284.4  748.68
     304  748.38   313.8  748.48   323.7  749.45   333.5  753.78   362.9  771.26
   382.5  782.53   411.9   799.2   431.6  810.81   441.4  816.78   451.2  822.61
     461  828.27   470.8  833.79   480.6  839.11     510   854.2   539.4  867.65
#Mann= 3 , 0 , 0
       0      .1       0   284.4    .045       0   323.7      .1       0
Bank Sta=284.4,323.7
XS Rating Curve= 0 ,0
Exp/Cntr=0.3,0.1

Type RM Length L Ch R = 1 ,43431   ,390.1,393.9,397.6
XS GIS Cut Line= 4
     1869760.521      516528.574     1870321.919      516717.766
     1870532.327      516698.709      1870888.23      516794.195
#Sta/Elev= 30
       0   812.4    48.6   802.3      68  796.53   126.2  776.48   145.7  771.55
   165.1  768.29   233.1  759.83   398.2  753.04   407.9  751.02   417.6  747.54
   446.7   746.6   456.4  746.66   466.2  748.26   475.9  753.72   514.7  784.64
   534.2  798.69     573  825.02   611.6  847.25   630.8  856.91   678.8  878.29
   765.3  913.09   803.7  932.22   813.4  932.37   842.5  928.61     920  913.81
   939.4  911.42   958.8     911   997.6  917.17  1123.7   952.3  1172.2  969.11
#Mann= 3 , 0 , 0
       0      .1       0   417.6    .045       0   456.4      .1       0
Bank Sta=417.6,456.4
XS Rating Curve= 0 ,0
Exp/Cntr=0.3,0.1

Type RM Length L Ch R = 1 ,43037.2 ,148.3,173.8,199.3
XS GIS Cut Line= 3
      1869765.43       516885.68     1870220.717      517129.367
     1870430.044      517473.128
#Sta/Elev= 30
       0  786.17    19.5  779.05    68.2  757.41      78  754.26    97.4  753.25
   272.8  754.74   282.6  754.42   292.3  752.21     302  748.24   311.8  746.13
   321.5   745.9     341  746.22   350.8  749.03   360.5  754.04   399.5  776.23
   496.9  825.72   506.7  830.37   516.4  834.03   526.2  838.69     536  842.45
   565.5  854.87   575.3  858.35   604.8  867.39     644  880.96   712.7  899.26
   761.8  911.55   791.3  917.75   879.6  933.05   899.2  935.65   918.9  937.11
#Mann= 3 , 0 , 0
       0      .1       0   311.8    .045       0     341      .1       0
Bank Sta=311.8,341
XS Rating Curve= 0 ,0
Exp/Cntr=0.3,0.1

Type RM Length L Ch R = 1 ,42863.4 ,61.7,63.3,64.8
XS GIS Cut Line= 4
     1869739.053         516996.     1869939.747      517092.528
     1869964.078      517309.191     1870068.914      517359.889
#Sta/Elev= 30
       0  790.76     9.7   787.5    19.4  784.06      29  780.34    38.7  776.14
    48.4  771.54    58.1  766.39    67.8  760.43    77.5  755.53    87.1  753.18
    96.8  752.73   116.2   752.7   222.7  751.81   251.1  751.06   260.6  750.45
   270.1  749.23   279.6  747.64   289.1  746.26   298.5  745.52   316.6  745.34
     327  745.48   345.9  745.48   355.4  746.33   364.9  748.97   374.4  752.09
   383.8  754.52   402.8  758.31   440.7  768.07   469.8  785.69   557.2  837.92
#Mann= 3 , 0 , 0
       0      .1       0   298.5    .045       0     327      .1       0
Bank Sta=298.5,327
XS Rating Curve= 0 ,0
Exp/Cntr=0.3,0.1

Type RM Length L Ch R = 1 ,42800.1 ,493.2,469.5,445.7
XS GIS Cut Line= 4
     1869728.123      517064.499     1869900.164      517145.305
     1869926.515      517379.954     1870022.386      517428.639
#Sta/Elev= 30
       0  791.69     9.5  788.12      19  784.14    28.5  779.81      38  775.04
    47.5  769.58    66.5  757.64      76  753.68    85.5  752.34   190.1  749.99
   199.9   749.5   219.6  749.03   229.4  748.45   249.1  746.09   258.9  745.48
   278.6  745.21   288.5  745.38   298.3  745.31   308.1  745.67     318  747.36
   327.8  749.91   337.6  751.77   347.5  752.43   367.2  752.83   386.8   753.7
   396.7  754.84   406.5  756.72   426.2  761.26   475.1   789.3   533.7  822.53
#Mann= 3 , 0 , 0
       0      .1       0   258.9    .045       0   288.5      .1       0
Bank Sta=258.9,288.5
XS Rating Curve= 0 ,0
Exp/Cntr=0.3,0.1

Type RM Length L Ch R = 1 ,42330.6 ,556.9,559.6,562.1
XS GIS Cut Line= 3
     1869477.097      517489.074     1869817.693      517742.633
     1869982.305      517970.845
#Sta/Elev= 30
       0   825.4    67.6  791.34    96.5  777.69   106.2  771.98   135.1  751.82
   144.8  746.61   154.4  744.59   164.1  744.31   183.4   744.9     193  747.24
   202.7  748.92   212.3  748.89   231.6   747.8   260.6  747.74   318.5  751.72
   347.4  752.65   424.6  753.64   511.9  753.26   521.6  753.39   531.4  754.94
     541   759.5   550.8  765.63     609  806.95   618.7  813.48   638.1  825.33
   647.8  830.69   657.5  834.92   667.2  838.38   686.6  844.43     706  849.19
#Mann= 3 , 0 , 0
       0      .1       0   144.8    .045       0   183.4      .1       0
Bank Sta=144.8,183.4
XS Rating Curve= 0 ,0
Exp/Cntr=0.3,0.1

Type RM Length L Ch R = 1 ,41771.1 ,446.7,446.6,446.4
XS GIS Cut Line= 2
     1869119.024      517888.813     1869586.472      518328.918
#Sta/Elev= 30
       0  806.47    68.1  780.93    77.8   777.1    87.6  772.52    97.3  766.55
   126.5  747.92   136.2  742.69   145.9  740.75   155.6  740.46   165.4  740.93
   175.1  742.03   184.8  743.34   204.3  746.32     214  747.27   252.9   748.2
   262.6  748.27   359.9  747.32   389.1   747.6   408.6   747.6   437.8   747.2
   457.2   747.2   496.1  747.32     535  747.67   544.8  749.65   554.5  754.83
   593.4  782.05   612.8   795.1   622.6  801.08   632.3  805.92     642   810.3
#Mann= 3 , 0 , 0
       0      .1       0   136.2    .045       0   175.1      .1       0
Bank Sta=136.2,175.1
XS Rating Curve= 0 ,0
Exp/Cntr=0.3,0.1

Type RM Length L Ch R = 1 ,41324.4 ,234.5,231.5,228.7
XS GIS Cut Line= 3
     1868833.651       518218.24     1869112.514      518473.232
     1869178.703      518560.037
#Sta/Elev= 30
       0   783.7    19.4  775.39    29.1  771.36    58.1  759.05    67.8  754.82
    77.5  751.03    87.2   748.6    96.9  748.28     126  748.14     155  747.89
   174.4  747.84   193.8  747.62   203.5  746.43   213.2  743.08   222.8  739.88
   232.5  738.71   242.2   738.7   251.9  738.74   261.6  739.43   271.3  742.46
     281  745.16   290.7  746.32   339.1   748.2   368.2  749.42   414.3  751.56
   423.4  753.05   432.4  756.42   441.6  761.24   459.7  771.72     487  787.81
#Mann= 3 , 0 , 0
       0      .1       0   222.8    .045       0   261.6      .1       0
Bank Sta=222.8,261.6
XS Rating Curve= 0 ,0
Exp/Cntr=0.3,0.1

Type RM Length L Ch R = 1 ,41092.9 ,298.4,301.1,303.6
XS GIS Cut Line= 2
      1868657.87      518403.787     1869044.154      518677.225
#Sta/Elev= 30
       0  800.77    19.3  788.22    38.6   775.8    67.6  757.52    77.3  751.82
    86.9  748.12    96.6  747.42   106.2  747.24   144.9  746.69   173.8  746.38
   231.8  745.91   251.1  745.49   280.1  745.14   299.4  744.67   309.1  743.34
   318.7  740.44   328.4  738.76     338  738.61   347.7  738.75   357.4  740.12
     367  743.41   386.3  751.56     396  755.86   405.7   760.4   415.3   764.3
     425  766.74   444.3  770.34     454  772.74   463.6   775.5   473.3  778.43
#Mann= 3 , 0 , 0
       0      .1       0   318.7    .045       0   357.4      .1       0
Bank Sta=318.7,357.4
XS Rating Curve= 0 ,0
Exp/Cntr=0.3,0.1

Type RM Length L Ch R = 1 ,40791.8 ,194.3,177.3,160.2
XS GIS Cut Line= 3
     1868533.087       518603.44     1868784.823      518829.135
     1869009.432      518848.666
#Sta/Elev= 30
       0  818.18     9.7  815.75    19.3  812.31      29  808.46    38.6  803.97
    48.3  799.01      58  793.71    67.6  788.02   115.9  758.42   125.6  753.03
   135.2  748.01   144.9  743.25   154.6  739.92   164.2  738.56   202.9   738.2
   212.5  738.25   222.2  738.72   231.8  739.33   241.5  740.64   251.2  743.68
   260.8  747.11   270.5  748.22   406.7  749.15   445.9  750.46   465.5  750.69
   475.3  751.09   485.1  752.33   494.9  754.38   534.2  763.98   563.6  772.25
#Mann= 3 , 0 , 0
       0      .1       0   164.2    .045       0   222.2      .1       0
#XS Ineff= 2 , 0
                          331.02          757.17
Permanent Ineff=
       F       F
Bank Sta=164.2,222.2
XS Rating Curve= 0 ,0
Exp/Cntr=0.3,0.1

Type RM Length L Ch R = 1 ,40614.5 ,81.4,80.4,79.4
XS GIS Cut Line= 3
     1868565.639      518895.324     1868751.186      518892.069
      1868981.22      518864.942
#Sta/Elev= 29
       0  765.61     9.8  765.92    19.5  765.12    29.3  760.64    39.1  753.11
    48.8  745.84    58.6  740.49    68.4   738.4    87.9  738.03    97.7  738.84
   107.4  742.45   117.2  746.27     127  747.72     166  748.83   185.6  749.12
   204.9   749.3   262.8  749.34   272.4  748.09   282.1  747.77   291.7  747.91
   301.4  748.38   320.7  750.08     340  751.32   349.6  751.78     369  752.36
   378.6  753.27   388.2  755.18   397.9  757.65   417.2  762.98
#Mann= 3 , 0 , 0
       0      .1       0    58.6    .045       0    97.7      .1       0
#XS Ineff= 2 , 0
                          225.21          753.55
Permanent Ineff=
       F       F
Bank Sta=58.6,97.7
XS Rating Curve= 0 ,0
Exp/Cntr=0.3,0.1

Type RM Length L Ch R = 1 ,40534.2 ,77.8,77.8,77.9
XS GIS Cut Line= 5
     1868573.802      518978.812     1868722.034      518969.157
     1868785.643      518975.404      1868827.67      518987.331
     1868960.567       519070.25
#Sta/Elev= 30
       0  757.24     9.3  757.17    27.8  756.56    37.1  753.97    46.4  748.58
    55.7  742.42    62.6739.7342      65   738.8    74.3  737.88    83.6  737.81
    92.8  739.03   111.4  745.63   120.7  747.49     130  748.22   175.9  750.01
   203.3  750.09   221.2  749.75   229.9  749.34   238.7  748.44   256.2  745.16
   265.9  747.51   275.7  748.42   305.1  748.74   314.9  748.64   344.3  747.75
   363.8  748.05   373.6  748.43   383.4  748.42   393.2  748.93   412.8  749.47
#Mann= 3 , 0 , 0
       0      .1       0    62.6    .045       0    92.8      .1       0
#XS Ineff= 2 , 0
                          192.99          753.08
Permanent Ineff=
       F       F
Bank Sta=62.6,92.8
XS Rating Curve= 0 ,0
Exp/Cntr=0.3,0.1

Type RM Length L Ch R = 1 ,40456.4 ,187.3,210.7,232.9
XS GIS Cut Line= 5
     1868605.696      519053.443     1868722.602      519045.829
     1868786.211      519052.076     1868828.238      519064.003
     1868961.135      519146.922
#Sta/Elev= 30
       0  750.94     9.8  750.89    19.5   749.2    29.3  745.27      39  740.77
    48.8   738.2    58.6   737.7    68.3  738.15    69.4738.4172    78.1  740.53
    87.9  744.41    97.6  746.23   107.4  746.28   117.2     746   126.3  745.55
   162.8  744.23   171.9  743.62   189.8  742.71   198.5  742.71   207.3  742.87
   224.8  743.42   234.6  744.19   244.3  745.04   254.1  746.27   263.9  747.64
   283.5  749.26   293.3  749.84   312.9  750.73   361.8  752.24   381.4  753.05
#Mann= 3 , 0 , 0
       0      .1       0    48.8    .045       0    69.4      .1       0
#XS Ineff= 2 , 0
                          124.65          749.02
Permanent Ineff=
       F       F
Bank Sta=48.8,69.4
XS Rating Curve= 0 ,0
Exp/Cntr=0.3,0.1

Type RM Length L Ch R = 1 ,40245.7 ,420.2,453.3,487.4
XS GIS Cut Line= 4
      1868593.85      519075.445     1868610.126      519176.357
     1868705.081      519298.298     1868720.804      519425.923
#Sta/Elev= 30
       0     749     9.3  748.59    46.5   747.8    83.6  747.65    92.9  747.39
   111.9  746.41   121.5  746.58   131.2  745.19   140.8   743.3   150.5  741.76
   160.2  740.57   169.8  739.09   179.5   737.3   189.2   736.2   208.5  736.13
   218.1  737.05   227.8  740.62   256.8  755.36     266  759.39   275.1  763.66
   284.3  768.35   293.5  773.52   302.7  779.19   311.9  785.34   321.1   791.9
   330.2  798.88   348.6  813.63   357.8  820.44     367  826.83   385.4   839.2
#Mann= 3 , 0 , 0
       0      .1       0   189.2    .045       0   218.1      .1       0
Bank Sta=189.2,218.1
XS Rating Curve= 0 ,0
Exp/Cntr=0.3,0.1

Type RM Length L Ch R = 1 ,39792.3 ,303.1,308.6,314
XS GIS Cut Line= 4
     1868518.981      518864.942     1868239.311      519116.747
     1868224.927      519276.183     1868299.797      519473.666
#Sta/Elev= 30
       0  766.04      29  758.07    48.2  754.53    57.9  751.34    67.6  749.16
    77.2  748.35   241.2  746.21   250.9  745.46   260.5  742.55   270.2   737.6
   279.8  734.44   308.8  732.72   318.4  736.77   385.7  785.73   395.2   793.1
     414  810.07   423.4  817.47   432.8   823.6   442.2  828.63   461.1  836.59
   498.7  848.72   517.6   856.6     546  874.78   574.8  887.74   603.6  905.43
   622.8  914.87   632.4  918.72   661.2  927.79   680.4  932.57   747.6   946.5
#Mann= 3 , 0 , 0
       0      .1       0   270.2    .045       0   318.4      .1       0
Bank Sta=270.2,318.4
XS Rating Curve= 0 ,0
Exp/Cntr=0.3,0.1

Type RM Length L Ch R = 1 ,39483.8 ,302.2,311.2,320
XS GIS Cut Line= 5
     1868381.177      518608.865     1868184.451      518781.788
     1867977.414       518892.79     1867846.827      519022.864
     1867712.774      519190.463
#Sta/Elev= 30
       0  784.43    19.4  781.53    38.8  776.01    48.5  771.28    87.3  746.53
      97  742.05   106.7  741.23   126.1   741.1   301.1  744.61   310.9  742.64
   330.4  732.26   340.2  730.12     350  730.62   369.6  734.01   379.4  738.79
     399  750.27   418.5  760.58   467.5  783.19   496.8  795.69   535.6  810.98
   574.4  828.06   613.2  840.09     652  856.66   671.4  863.65   681.2   866.6
   720.2  875.47   788.5  888.46   856.8  904.76   876.3  908.45   895.8  911.15
#Mann= 3 , 0 , 0
       0      .1       0   330.4    .045       0   369.6      .1       0
#XS Ineff= 2 , 0
          294.62  759.17
Permanent Ineff=
       F       F
Bank Sta=330.4,369.6
XS Rating Curve= 0 ,0
Exp/Cntr=0.3,0.1

Type RM Length L Ch R = 1 ,39172.6 ,506,491.6,477.2
XS GIS Cut Line= 4
     1868280.265      518439.595     1868128.356      518515.549
     1867973.191       518530.74     1867879.875      518574.143
#Sta/Elev= 30
       0  784.67     9.4  780.83    18.9  777.33    28.3  774.49    56.6  767.22
      66  762.65    75.5  755.77    84.9  747.91    94.4  741.89   103.8   740.3
   122.7  741.15   179.6  740.89   218.6  740.43   228.3  738.09     238  733.81
   247.8  731.04   257.5  730.22   267.3  730.01     277  731.46   286.8  739.03
   296.5  747.81   306.3  755.19     316  760.49   325.8  764.01   335.1  767.07
   372.5  778.65   381.9  782.02   400.6  789.08     410  792.75   428.7  800.58
#Mann= 3 , 0 , 0
       0      .1       0   247.8    .045       0     277      .1       0
Bank Sta=247.8,277
XS Rating Curve= 0 ,0
Exp/Cntr=0.3,0.1

Type RM Length L Ch R = 1 ,38681   ,311.2,293.5,275.9
XS GIS Cut Line= 3
     1868128.356      517906.826     1867839.727      518166.157
     1867787.644      518300.706
#Sta/Elev= 30
       0  852.31     9.7  851.88    29.1  848.56    38.8  846.06    48.5  841.97
    58.2  837.22    67.9  831.61    77.6  825.16   116.4  797.05   135.8  784.77
   145.5  779.49   155.2  775.61   174.6  771.61   184.3  764.24     194   750.9
   203.7  738.68   211.9732.2975   213.4  731.13   223.1  729.82   232.8  730.24
   242.5   731.9   261.9  733.38   271.6  737.38   281.3  740.53     291  741.64
   358.9  742.85   484.2   741.6   493.8  742.76   513.1  747.45   532.3  750.71
#Mann= 3 , 0 , 0
       0      .1       0   211.9    .045       0   242.5      .1       0
#XS Ineff= 2 , 0
                          348.44           751.5
Permanent Ineff=
       F       F
Bank Sta=211.9,242.5
XS Rating Curve= 0 ,0
Exp/Cntr=0.3,0.1

Type RM Length L Ch R = 1 ,38387.4 ,414.9,391.5,368
XS GIS Cut Line= 4
     1867767.028      517606.261      1867730.63      517804.667
     1867710.371      518130.497     1867717.124      518300.164
#Sta/Elev= 30
       0  783.36    38.4  776.12    76.8  770.61    86.4  768.02   105.7  760.89
   115.3  758.49   124.9   758.3   144.1  761.48   153.7  762.48   172.9  762.69
   182.5  762.35   192.1  761.32   201.7  758.99   220.9  751.92   259.3  735.71
   268.9  730.97   278.5  728.91   288.1  728.59   307.3  728.99   316.9  731.43
   336.1  737.62   345.7  739.48   355.3  740.14   403.4  740.67   451.4   742.6
   499.4  743.76   631.9  743.12   641.4  743.56   650.8  744.77     698  751.79
#Mann= 3 , 0 , 0
       0      .1       0   268.9    .045       0   316.9      .1       0
Bank Sta=268.9,316.9
XS Rating Curve= 0 ,0
Exp/Cntr=0.3,0.1

Type RM Length L Ch R = 1 ,37996   ,259.2,262.1,265.1
XS GIS Cut Line= 3
     1867324.609      518035.955     1867512.847      518161.729
     1867609.921       518342.37
#Sta/Elev= 30
       0   794.2     9.4  791.51    18.9  787.29    28.3  782.94    37.7   778.4
    47.2  773.62    94.3  747.93   103.8  742.98   113.2  738.24   122.6  733.68
   132.1  730.02   141.5  728.53   150.9   728.4   160.4  728.48   169.8  728.16
   179.2  727.65   188.7  727.95   198.1  731.98   207.5  738.05     217  740.64
   226.4  741.04   245.9  740.85     285  739.54   304.5  739.19     324  739.32
   333.8  739.94   343.6  741.58   382.6  749.77   402.2  753.67   431.5  760.58
#Mann= 3 , 0 , 0
       0      .1       0   160.4    .045       0   188.7      .1       0
Bank Sta=160.4,188.7
XS Rating Curve= 0 ,0
Exp/Cntr=0.3,0.1

Type RM Length L Ch R = 1 ,37733.8 ,392.5,430.9,469.3
XS GIS Cut Line= 4
     1867195.459       518155.82     1867219.938      518263.867
     1867383.697      518407.368     1867394.671      518560.997
#Sta/Elev= 30
       0  758.52    27.7  752.19    36.9   750.7    46.2  749.66   110.8  744.58
   139.2  743.25   158.1  741.45   167.6  740.02     177  738.16   186.5  735.66
   205.4  729.62   214.9  728.47   224.4   728.2   243.3  728.28   252.8  729.84
   262.2  732.83   271.7  734.37   281.2  736.68   290.7   741.9   300.1  747.57
   319.1  757.65   328.5  762.22   338.2  766.24   347.8  769.64     367  775.59
   424.8   792.5   453.7   801.5   463.3  805.47   472.9   810.7   482.5  816.41
#Mann= 3 , 0 , 0
       0      .1       0   205.4    .045       0   252.8      .1       0
Bank Sta=205.4,252.8
XS Rating Curve= 0 ,0
Exp/Cntr=0.3,0.1

Type RM Length L Ch R = 1 ,37302.9 ,581.2,571.5,561.8
XS GIS Cut Line= 3
     1867052.802      518008.943     1867018.194      518217.441
     1866780.206      518430.385
#Sta/Elev= 30
       0  807.02    28.8  791.93    57.6  775.56    76.8  765.06    96.1  755.65
   105.7  751.47   115.3  748.01   124.9  746.12   144.1  745.11   163.3  744.72
   211.4  745.04   230.7  743.48   250.1  741.08   269.4  737.78   279.1   734.7
   288.8  730.12   298.4  728.26   308.1   728.1   317.8  728.13   327.5  729.58
   366.2  742.52   385.5  750.32   404.9  758.86   414.6   763.5   433.9  773.71
     463  790.69     492  807.13   511.3  817.33     521  822.04   530.7  826.28
#Mann= 3 , 0 , 0
       0      .1       0   288.8    .045       0   327.5      .1       0
Bank Sta=288.8,327.5
XS Rating Curve= 0 ,0
Exp/Cntr=0.3,0.1

Type RM Length L Ch R = 1 ,36731.4 ,321.7,327.4,333.1
XS GIS Cut Line= 3
     1866664.508      517724.475     1866574.187       517840.12
     1866438.284      518149.067
#Sta/Elev= 30
       0  863.46    29.4  849.85    58.7  836.02    68.5  830.78    78.3  823.55
   117.4   787.8   127.2  778.95   146.7  761.72     166  745.91   175.7  739.85
   185.3  736.37     195  734.04   214.2  729.59   223.9  728.34   243.2  727.42
   252.8  727.51   262.5  728.75   281.7     732     301  734.56   310.7  735.63
   320.3  736.51   339.6  737.84   349.2  738.14   368.5  738.34   378.2   739.8
   387.8  744.29   397.5  750.48   426.4  769.46     436  775.27   484.2  801.29
#Mann= 3 , 0 , 0
       0      .1       0   223.9    .045       0   262.5      .1       0
Bank Sta=223.9,262.5
XS Rating Curve= 0 ,0
Exp/Cntr=0.3,0.1

Type RM Length L Ch R = 1 ,36403.9 ,434.1,440.8,447.4
XS GIS Cut Line= 2
     1866387.158      517605.792     1866156.045       517898.66
#Sta/Elev= 30
       0  823.95    29.4  804.54    49.1  791.78    68.7  779.22    88.4  766.82
     108  754.75   117.8   748.8   127.6  743.04   137.4  738.77   147.3  736.69
   157.1  735.83   186.5  733.67   196.4  732.74   206.2   731.2     216  728.75
   225.8  726.94   235.6  726.43   245.4  726.62   255.3  727.86   265.1  731.97
   274.9  737.15   284.7  742.66   294.5  748.73   304.4  755.07   314.2  761.47
     324  767.65   333.8  773.58   353.4  784.78   363.3  790.21   373.1  795.72
#Mann= 3 , 0 , 0
       0      .1       0   225.8    .045       0   255.3      .1       0
Bank Sta=225.8,255.3
XS Rating Curve= 0 ,0
Exp/Cntr=0.3,0.1

Type RM Length L Ch R = 1 ,35963.2 ,536.3,534.1,531.9
XS GIS Cut Line= 2
     1866181.942      517306.763     1865844.835      517540.387
#Sta/Elev= 25
       0  848.92     9.8     843    19.5  835.96    39.1  820.87    58.6  805.67
    97.6  775.54   117.2  760.71     127  753.35   136.7  746.19   146.5  740.35
   156.2  738.25     166  737.32   224.6  732.26   234.4  731.06   244.1  728.98
   253.9  726.13   263.7  724.29   273.4  724.12   283.2  724.32     293   724.4
   302.7   726.9   322.3  736.86   351.6  752.07   380.8  767.36   410.2  782.21
#Mann= 3 , 0 , 0
       0      .1       0   263.7    .045       0     293      .1       0
Bank Sta=263.7,293
XS Rating Curve= 0 ,0
Exp/Cntr=0.3,0.1

Type RM Length L Ch R = 1 ,35429.1 ,402.4,388.4,373.9
XS GIS Cut Line= 3
     1866070.952      516751.545     1865858.739      516865.485
     1865539.708      517134.668
#Sta/Elev= 30
       0   873.9    38.5  859.06    67.4  848.53    86.7  840.88    96.4  837.78
     106  835.11   144.5  827.92   173.4  820.46   221.6  809.51   289.4  791.32
   308.8  785.62   347.6  771.65   357.4  765.88   367.1  758.19   376.8  751.72
   386.5  747.06   425.3   734.8   444.7  726.16   454.4  723.11   464.1  722.07
   473.8  723.67   493.3  722.55     503  725.36   512.7  731.25   522.4  733.79
   561.2  736.96   570.9  739.09   580.6  742.99   629.2   764.8   658.3  776.58
#Mann= 3 , 0 , 0
       0      .1       0   454.4    .045       0   493.3      .1       0
Bank Sta=454.4,493.3
XS Rating Curve= 0 ,0
Exp/Cntr=0.3,0.1

Type RM Length L Ch R = 1 ,35040.7 ,303.4,285.5,267.6
XS GIS Cut Line= 4
     1865405.829      516600.575     1865347.435      516829.879
     1865310.404      516980.849     1865316.101      517047.789
#Sta/Elev= 30
       0  784.45     9.5  780.73    28.4  772.96    47.3  764.46    56.8  759.41
    66.2  752.38    75.7  744.73    85.2   740.6    94.6  739.82   151.4  737.47
   236.6  733.36     256  732.98   265.8  732.34   275.5  730.19   285.2  726.16
   294.9  722.48   304.6  721.15   314.3     721   324.1     721   333.8  721.97
   343.5  727.37   353.2   737.2   362.9  746.16   372.6  750.92   382.4  752.62
   392.1  753.77   411.3  758.28   430.5  762.25   449.6  765.92   459.2  767.43
#Mann= 3 , 0 , 0
       0      .1       0   294.9    .045       0   333.8      .1       0
Bank Sta=294.9,333.8
XS Rating Curve= 0 ,0
Exp/Cntr=0.3,0.1

Type RM Length L Ch R = 1 ,34755.2 ,348.7,322.5,296.3
XS GIS Cut Line= 4
     1864870.312      516658.969     1865025.555      516811.364
     1865125.252      516975.152      1865261.98       517054.91
#Sta/Elev= 30
       0  926.53    37.8  897.71    85.1   862.4     104  847.84   113.5  840.26
   132.4  824.77   141.9  816.57   160.8  799.74   179.7  781.97   189.2  772.82
   217.5  744.37   227.1  736.63   236.7  731.74   246.3  727.78   255.9  724.16
   263.3722.1404   265.5  721.54   275.1     721   284.6     721   294.2  721.37
   303.8  723.26     323  729.06   332.6  731.23   342.2  732.27   409.3  734.42
     521  736.57   530.3  737.57   539.6  739.99     549   743.5   567.6  750.84
#Mann= 3 , 0 , 0
       0      .1       0   263.3    .045       0   294.2      .1       0
Bank Sta=263.3,294.2
XS Rating Curve= 0 ,0
Exp/Cntr=0.3,0.1

Type RM Length L Ch R = 1 ,34432.7 ,413.6,409.8,405.9
XS GIS Cut Line= 3
     1864870.312      517191.638     1865136.646      517156.031
       1865254.8      517146.718
#Sta/Elev= 30
       0  846.18     9.6  839.97    19.2  833.35    28.8  826.25    38.4  818.76
      48  810.75    57.6  802.33    67.2  793.51    76.8  784.42      96  766.02
   105.6  756.92   115.2  748.03   124.8  739.38   134.4  730.96     144  724.15
   153.5  721.19   163.1     721   182.3     721   191.9  721.26   201.5  723.45
   211.1  729.68   220.7  734.03   230.3   734.1   286.9   734.1   314.3     734
   350.8  734.03   359.9  734.49     369  736.67   378.1  740.65   387.2  744.83
#Mann= 3 , 0 , 0
       0      .1       0   153.5    .045       0   191.9      .1       0
Bank Sta=153.5,191.9
XS Rating Curve= 0 ,0
Exp/Cntr=0.3,0.1

Type RM Length L Ch R = 1 ,34022.9 ,544.6,563,581.3
XS GIS Cut Line= 3
     1865008.464      517604.669     1865224.704      517536.999
     1865417.385      517521.409
#Sta/Elev= 30
       0  775.59    18.9  766.13    37.8   756.5    56.6  746.75    66.1     742
    75.5   737.2      85  732.66    94.4   729.2   103.8  725.26   113.3  721.86
   122.7  721.05     151   720.9   160.5  721.13   169.9  722.43   179.4  724.73
   188.8  726.31   226.6  728.22   245.9  728.95   274.9  730.32   284.6  731.02
   294.2  733.58   303.9  738.46   313.6  744.03   332.9  755.34   342.6  760.89
   352.2   766.2   371.6  776.42   381.2   781.8   390.9   787.4   419.9  804.45
#Mann= 3 , 0 , 0
       0      .1       0   113.3    .045       0   160.5      .1       0
Bank Sta=113.3,160.5
XS Rating Curve= 0 ,0
Exp/Cntr=0.3,0.1

Type RM Length L Ch R = 1 ,33459.9 ,360.6,385.2,409.8
XS GIS Cut Line= 3
     1864933.483      517947.627     1865447.806         518233.
     1865605.141       518380.57
#Sta/Elev= 30
       0  755.14      49  733.37    58.8  729.51    68.6  727.41   137.2  728.33
   205.9  728.18   215.7  727.28   245.1  720.41   254.9  719.53   274.5   719.6
   284.3  720.68   294.1  725.34   303.9  733.04   362.7  776.88   382.3  790.42
   401.9  803.12   421.5  814.16   470.6  838.82     500  854.61   529.4  871.75
   558.8  890.82   568.6  896.72   578.4  901.32   588.2  903.33     598   903.1
   656.8  899.28   705.8  894.19   784.3  885.11   794.1  883.58   803.9  881.11
#Mann= 3 , 0 , 0
       0      .1       0   245.1    .045       0   284.3      .1       0
#XS Ineff= 2 , 0
          162.89  740.42
Permanent Ineff=
       F       F
Bank Sta=245.1,284.3
XS Rating Curve= 0 ,0
Exp/Cntr=0.3,0.1

Type RM Length L Ch R = 1 ,33074.7 ,507.6,517.7,527.2
XS GIS Cut Line= 3
     1864840.167      517989.945     1864877.059       518155.96
     1864871.634      518444.589
#Sta/Elev= 30
       0  770.05    18.9  762.17    37.8  753.84    47.2  749.46    56.7   745.2
    66.1  741.34    75.6  737.84      85  734.55    94.5  731.41   103.9  728.87
   113.4  727.72   151.2  727.56   179.7  727.25   189.3  727.11   198.9  726.59
   208.6  725.47   237.4  720.94     247  719.54   256.7  718.66   266.3   718.4
   304.8   718.4   314.4  720.37     324   726.8   333.6   734.6   343.3  741.38
   372.1   760.1   381.8   766.2     401  777.95   410.6  784.01   458.7  815.55
#Mann= 3 , 0 , 0
       0      .1       0   256.7    .045       0   304.8      .1       0
Bank Sta=256.7,304.8
XS Rating Curve= 0 ,0
Exp/Cntr=0.3,0.1

Type RM Length L Ch R = 1 ,32557.1 ,352.2,354.1,355.8
XS GIS Cut Line= 4
      1864494.03       517916.16     1864338.865      518234.085
     1864449.542      518390.335     1864460.393      518522.714
#Sta/Elev= 30
       0   754.2    19.6  745.32    29.5  741.97    68.8  731.69    78.6  729.82
    88.4  728.87    98.3  728.47     226  724.28   235.8  722.64   255.5  714.25
   265.3  712.51     285  712.84   294.8  714.31   304.6  720.23   314.5  729.62
   324.3  738.41   334.1  746.86   343.9  754.53   353.8  759.55   372.9  766.72
   401.6  775.77   411.2  779.68   439.9  792.73   459.1   799.6   478.2  803.98
   526.1  812.03   545.2  816.02   621.1   819.6   659.1   820.5   678.1  820.25
#Mann= 3 , 0 , 0
       0      .1       0   255.5    .045       0   294.8      .1       0
Bank Sta=255.5,294.8
XS Rating Curve= 0 ,0
Exp/Cntr=0.3,0.1

Type RM Length L Ch R = 1 ,32203   ,632.3,635.8,639.3
XS GIS Cut Line= 3
      1864233.92      517704.066     1864002.493      518095.197
     1863833.223      518280.743
#Sta/Elev= 30
       0  780.76      29   764.8    48.4  754.86    96.7  734.41   106.4  731.39
     116  729.99   135.4  727.93     174  724.34   183.7  723.78   290.1  723.55
   299.8  721.77   309.4  715.69   319.1  711.97   328.8  711.13   338.4  711.12
   348.1  711.76   357.8  715.24   386.8   735.1   425.5  762.86   435.1  768.93
   444.8  773.23   454.5  776.65   541.4  805.59   551.1  809.41   570.4  817.88
   628.4  844.23     638  847.57   647.7  853.34   686.3  879.09   705.6  891.29
#Mann= 3 , 0 , 0
       0      .1       0   319.1    .045       0   348.1      .1       0
#XS Ineff= 2 , 0
          266.29     736
Permanent Ineff=
       F       F
Bank Sta=319.1,348.1
XS Rating Curve= 0 ,0
Exp/Cntr=0.3,0.1

Type RM Length L Ch R = 1 ,31567.2 ,371.9,358.2,344.6
XS GIS Cut Line= 4
     1863684.568      517246.672     1863688.908      517462.601
     1863493.596      517698.061     1863470.809       517834.78
#Sta/Elev= 30
       0  845.72    29.4  834.96    68.7  817.95    88.4  809.01   117.8  794.93
   137.4  784.53   157.1  774.68   166.9  770.41   196.3   759.4   206.2  755.13
   225.5  742.55   235.1  736.94   244.6  733.13   282.9  720.43     302  712.88
   311.6   711.4   321.1   711.1   340.2  711.16   349.8  711.77   378.5  717.07
     388  717.98   445.4  719.66   474.1  721.04   483.6   721.8   493.2  723.87
   502.8  728.09   521.9  737.53   595.8  777.68   605.1  782.24   660.5  803.74
#Mann= 3 , 0 , 0
       0      .1       0     302    .045       0   349.8      .1       0
Bank Sta=302,349.8
XS Rating Curve= 0 ,0
Exp/Cntr=0.3,0.1

Type RM Length L Ch R = 1 ,31208.9 ,599.6,584.6,569.4
XS GIS Cut Line= 3
     1863364.473      517144.676     1863301.539      517317.202
     1863266.816      517704.572
#Sta/Elev= 30
       0  871.65    19.3  850.26      29  840.21    48.3   820.5      58  811.56
    67.7   804.7      87  793.44   106.3  782.75   125.6  772.61     145   762.7
   212.8  728.56   222.5  724.31   232.3  721.41   271.2  713.14   280.9  711.53
   290.6   711.1     310   711.1   319.8  711.41   329.5  713.29   339.2  716.75
   348.9  718.52     417  716.02   426.7  716.24   485.1  720.87   494.8  722.52
   504.5  725.93   514.2  729.82   533.7  736.88   562.8  746.81   572.6  751.16
#Mann= 3 , 0 , 0
       0      .1       0   280.9    .045       0   319.8      .1       0
Bank Sta=280.9,319.8
XS Rating Curve= 0 ,0
Exp/Cntr=0.3,0.1

Type RM Length L Ch R = 1 ,30624.3 ,357.2,349.6,341.9
XS GIS Cut Line= 2
     1862606.009      517320.457     1862896.808       517764.25
#Sta/Elev= 30
       0  837.72    19.6  824.74    39.3  812.04    49.1  806.53      59   801.6
    88.4  787.32    98.3  782.38   108.1  776.67   117.9  768.58   137.6  750.39
   147.4   741.1     167  722.81   176.9  714.81   186.7  711.48   196.5   711.1
     226   711.1   235.8  711.51   255.5  713.37   265.3  714.12   275.1  714.42
   304.6  714.49   324.2  714.68   432.3  716.89   442.2  718.19     452  722.15
   481.4  741.07   491.3   746.9   501.1  751.53   520.8  759.48   530.6  763.57
#Mann= 3 , 0 , 0
       0      .1       0   186.7    .045       0   235.8      .1       0
Bank Sta=186.7,235.8
XS Rating Curve= 0 ,0
Exp/Cntr=0.3,0.1

Type RM Length L Ch R = 1 ,30274.8 ,316.1,317.1,317.4
XS GIS Cut Line= 2
     1862358.613      517642.723     1862715.601      517915.075
#Sta/Elev= 25
       0  786.08     9.8  780.98    29.3  770.49      39  765.03    48.8  759.39
    58.6  753.48    68.3  746.24    78.1  735.55    87.8  722.58    97.6  714.09
   107.4  711.19   126.9   711.1   136.7  711.24   146.4   712.2   156.2  713.72
   165.9     715   175.7  715.94   185.5  716.59   302.6  719.98   351.4  721.56
   380.7  722.59   390.4   723.6   400.2  726.16   429.5  737.34     449  744.89
#Mann= 3 , 0 , 0
       0      .1       0    97.6    .045       0   146.4      .1       0
Bank Sta=97.6,146.4
XS Rating Curve= 0 ,0
Exp/Cntr=0.3,0.1

Type RM Length L Ch R = 1 ,29957.7 ,493.9,522,550.8
XS GIS Cut Line= 4
      1862222.98      517811.993      1862231.66      517928.096
     1862479.056      518122.323     1862520.289      518323.061
#Sta/Elev= 30
       0  758.82     9.7  756.18    19.4   753.1    87.3  729.93      97  727.23
   106.7  725.44   126.3  722.63   155.7  717.67   185.2  713.18   204.9  710.44
   214.7  710.21   250.2  710.13     254  710.13   263.9  711.05   293.4  716.17
   342.5  723.06   421.1  734.69     431  735.98   440.7  736.99     470  739.73
   479.8  741.09   489.5   742.9   499.3  745.59   518.8  753.67   528.5  757.47
   538.3   760.7   587.1  776.05   606.6  781.76   616.4  784.91   635.9  792.66
#Mann= 3 , 0 , 0
       0      .1       0   204.9    .045       0   263.9      .1       0
Bank Sta=204.9,263.9
XS Rating Curve= 0 ,0
Exp/Cntr=0.3,0.1
